--- EF_FEMA.prj (project) ---

Proj Title=East_Fork_FEMA
Current Plan=p11
Default Exp/Contr=0.3,0.1
English Units
Geom File=g01
Geom File=g02
Geom File=g03
Geom File=g04
Geom File=g05
Geom File=g06
Flow File=f01
Flow File=f02
Flow File=f03
Flow File=f04
Flow File=f05
Flow File=f06
Flow File=f07
Plan File=p01
Plan File=p02
Plan File=p03
Plan File=p04
Plan File=p05
Plan File=p06
Plan File=p07
Plan File=p08
Plan File=p09
Plan File=p10
Plan File=p11
Plan File=p12
Y Axis Title=Elevation
X Axis Title(PF)=Main Channel Distance
X Axis Title(XS)=Station
BEGIN DESCRIPTION:
East Fork Trinity River Existing Conditions Steady State Model
The With Levee run contains representation of all hydraulically significant levees held in place:
Kaufman MUD 1 - left bank, STA 39720-downstream limit, modeled with levee points
Kaufman 5 East - left bank, STA 53041-40855, modeled with levee points
Kaufman 5 West - right bank, STA 53041-46345, modeled with levee points
Kaufman LID 10 - right bank, STA 66590-53843, modeled with levee points
Kaufman LID 15 - left bank, STA 94766-70658, modeled with levee points
The Natural Valley (NV) run for each levee removes representation of that levee from the model geometry while holding all other levees in place:
Scenario G - NV run of Kaufman MUD 1 Levee
Scenario H - NV run ofKaufman 5 East Levee
Scenario I - NV run ofKaufman 5 West Levee
Scenario J - NV run ofKaufman LID 10 Levee
Scenario K - NV run ofKaufman LID 15 Levee
All field survey was based on NAVD88.
Stream Name: East Fork Trinity River
Study Extents: Lake Ray Hubbard dam to confluence with Trinity River
Date: April 2020
HEC-RAS v5.0.6
Prepared for: DHS/FEMA (Federal Emergency Management Agency)
Prepared by: Compass PTS JV
Contract #HSFE60-15-D-0003
Task Order #HSFE06-17-J-0047
END DESCRIPTION:
DSS File=dss
DSS Export Rating Curves= 0
DSS Export Rating Curve Sorted= 0
DSS Export Volume Flow Curves= 0
DXF Filename=..\..\..\..\..\..\HECRAS_506\_EastFork_Models_v506\test_terrain_tiles_.
DXF OffsetX= 0
DXF OffsetY= 0
DXF ScaleX= 1
DXF ScaleY= 10

--- EF_FEMA.p11 (plan) ---

Plan Title=EastFork_WithLevee
Program Version=5.06
Short Identifier=WithLevee
Geom File=g06
Flow File=f03
Subcritical Flow
K Sum by GR= 0
Std Step Tol= 0.01
Critical Tol= 0.01
Num of Std Step Trials= 20
Max Error Tol= 0.3
Flow Tol Ratio= 0.001
Split Flow NTrial= 30
Split Flow Tol= 0.02
Split Flow Ratio= 0.02
Log Output Level= 0
Friction Slope Method= 1
Unsteady Friction Slope Method= 2
Unsteady Bridges Friction Slope Method= 1
Parabolic Critical Depth
Global Vel Dist= 0 , 0 , 0
Global Log Level= 0
CheckData=True
Encroach Param=-1 ,0,0, 2
BEGIN DESCRIPTION:
Geometric data - All hydraulically significant non-accredited levees represented using levee points and IFAs
Flow data - Reduced discharges through Kaufman LID 15 based on With Levee supplemental model that used a lateral structure to represent the levee. Discharges also reduced from STA 9844-16998 based on supplemental With Levee model that used lateral structure to represent spill to the Trinity River with full discharges elsewhere.
END DESCRIPTION:
Computation Interval=1MIN
Output Interval=1HOUR
Instantaneous Interval=1HOUR
Mapping Interval=1HOUR
Computation Time Step Use Courant=        0
Computation Time Step Use Time Series=    0
Computation Time Step Count To Double=0
Computation Time Step Max Doubling=0
Computation Time Step Max Halving=0
Computation Time Step Residence Courant=0
Run HTab= 0
Run UNet= 0
Run Sediment= 0
Run PostProcess= 0
Run WQNet= 0
Run RASMapper= 0
UNET Theta= 1
UNET Theta Warmup= 1
UNET ZTol= 0.02
UNET ZSATol= 0.02
UNET MxIter= 20
UNET Max Iter WO Improvement= 0
UNET MaxInSteps= 0
UNET DtIC= 0
UNET DtMin= 0
UNET MaxCRTS= 20
UNET WFStab= 2
UNET SFStab= 1
UNET WFX= 1
UNET SFX= 1
UNET 1D Methodology=Finite Difference
UNET DSS MLevel= 4
UNET Pardiso=0
UNET DZMax Abort= 100
UNET Use Existing IB Tables=-1
UNET Froude Reduction=False
UNET Froude Limit= 0.8
UNET Froude Power= 4
UNET D1 Cores= 0
UNET D2 Coriolis=0
UNET D2 Cores= 0
UNET D2 Theta= 1
UNET D2 Theta Warmup= 1
UNET D2 Z Tol= 0.01
UNET D2 Volume Tol= 0.01
UNET D2 Max Iterations= 20
UNET D2 Equation= 0
UNET D2 RampUpFraction=0.1
UNET D2 TimeSlices= 1
UNET D2 BCVolumeCheck=0
UNET D1D2 MaxIter= 0
UNET D1D2 ZTol=0.01
UNET D1D2 QTol=0.1
UNET D1D2 MinQTol=1
DSS File=dss
Write IC File= 0
Write IC File at Fixed DateTime=0
Write IC File at Sim End=0
Echo Input=False
Echo Parameters=False
Echo Output=False
Write Detailed= 0
HDF Write Warmup=0
HDF Write Time Slices=0
HDF Flush=0
HDF Face Node Velocities=0
HDF Compression= 1
HDF Chunk Size= 1
HDF Spatial Parts= 1
HDF Use Max Rows=0
HDF Fixed Rows= 1
Calibration Method= 0
Calibration Iterations= 20
Calibration Max Change=0.05
Calibration Tolerance=0.2
Calibration Maximum=1.5
Calibration Minimum=0.5
Calibration Optimization Method= 1
WQ AD Non Conservative
WQ ULTIMATE=-1
WQ Max Comp Step=1HOUR
WQ Output Interval=15MIN
WQ Output Selected Increments= 0
WQ Output face flow=0
WQ Output face velocity=0
WQ Output face area=0
WQ Output face dispersion=0
WQ Output cell volume=0
WQ Output cell surface area=0
WQ Output cell continuity=0
WQ Output cumulative cell continuity=0
WQ Output face conc=0
WQ Output face dconc_dx=0
WQ Output face courant=0
WQ Output face peclet=0
WQ Output face adv mass=0
WQ Output face disp mass=0
WQ Output cell mass=0
WQ Output cell source sink temp=0
WQ Output nsm pathways=0
WQ Output nsm derived pathways=0
WQ Output MaxMinRange=-1
WQ Daily Max Min Mean=-1
WQ Daily Range=0
WQ Daily Time=0
WQ Create Restart=0
WQ Fixed Restart=0
WQ System Summary=0
WQ Write To DSS=0
WQ Use Fixed Temperature=0
Sorting and Armoring Iterations= 10
XS Update Threshold= 0.02
Bed Roughness Predictor= 0
Hydraulics Update Threshold= 0.02
Energy Slope Method= 1
Volume Change Method= 1
Sediment Retention Method= 0
XS Weighting Method= 0
Number of US Weighted Cross Sections= 1
Number of DS Weighted Cross Sections= 1
Upstream XS Weight=0
Main XS Weight=1
Downstream XS Weight=0
Number of DS XS's Weighted with US Boundary= 1
Upstream Boundary Weight= 1
Weight of XSs Associated with US Boundary= 0
Number of US XS's Weighted with DS Boundary= 1
Downstream Boundary Weight= 0.5
Weight of XSs Associated with DS Boundary= 0.5
Percentile Method= 0
Sediment Output Level= 3
Mass or Volume Output= 0
Output Increment Type= 1
Profile and TS Output Increment= 1
XS Output Flag= 0
XS Output Increment= 10
Write Gradation File= 0
Read Gradation Hotstart= 0
Write HDF5 File= 1
Write Binary Output= 1
Write DSS Sediment File= 0
SV Curve= 0
Specific Gage Flag= 0

--- EF_FEMA.p01 (plan) ---

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Plan Title=ScenarioG_EastFork_Kauf_MUD1_NV
Short Identifier=ScenarioG_NV
Geom File=g01
Flow File=f05
Optimized Weir=East Fork       ,1               ,18740
Geometric data - Kaufman MUD 1 as natural valley and all other hydraulically significant non-accredited levees represented using levee points and IFAs. Optimization turned on for lateral at confluence with Trinity River.
Flow data - Full discharges through Kaufman MUD 1 with reduced discharges through Kaufman LID 15 based on With Levee supplemental model that used a lateral structure to represent the levee

--- EF_FEMA.p02 (plan) ---

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Plan Title=ScenarioH_EastFork_Kauf_5_East_NV
Short Identifier=ScenarioH_NV
Geom File=g02
Flow File=f03
Encroach Param=-1 ,0,0, 0
Optimized Weir=East Fork       ,12030106000003  ,18740
Geometric data - Kaufman 5 East as natural valley and all other hydraulically significant non-accredited levees represented using levee points and IFAs
Flow data - Reduced discharges through Kaufman LID 15 based on With Levee supplemental model that used a lateral structure to represent the levee. Discharges also reduced from STA 9844-16998 based on the With Levee supplemental model that used lateral structure to represent spill to the Trinity River with full discharges elsewhere.

--- EF_FEMA.p03 (plan) ---

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Plan Title=ScenarioI_EastFork_Kauf_5_West_NV
Short Identifier=ScenarioI_NV
Geom File=g03
Flow File=f03
Encroach Param=-1 ,0,0, 0
Optimized Weir=East Fork       ,12030106000003  ,18740
Geometric data - Kaufman 5 West as natural valley and all other hydraulically significant non-accredited levees represented using levee points and IFAs
Flow data - Reduced discharges through Kaufman LID 15 based on With Levee supplemental model that used a lateral structure to represent the levee. Discharges also reduced from STA 9844-16998 based on With Levee supplemental model that used lateral structure to represent spill to the Trinity River with full discharges elsewhere.

--- EF_FEMA.p04 (plan) ---

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Plan Title=ScenarioJ_EastFork_Kauf_LID10_NV
Short Identifier=ScenarioJ_NV
Geom File=g04
Flow File=f03
Encroach Param=-1 ,0,0, 0
Optimized Weir=East Fork       ,12030106000003  ,18740
Geometric data - Kaufman LID 10 as natural valley and all other hydraulically significant non-accredited levees represented using levee points and IFAs
Flow data - Reduced discharges through Kaufman LID 15 based on With Levee supplemental model that used a lateral structure to represent the levee. Discharges also reduced from STA 9844-16998 based on With Levee supplemental model that used lateral structure to represent spill to the Trinity River with full discharges elsewhere.

--- EF_FEMA.p05 (plan) ---

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Plan Title=ScenarioK_EastFork_Kauf_LID15_NV
Short Identifier=ScenarioK_NV
Geom File=g05
Flow File=f01
Encroach Param=-1 ,0,0, 0
Optimized Weir=East Fork       ,12030106000003  ,18740
Geometric data - Kaufman LID 15 as natural valley and all other hydraulically significant non-accredited levees represented using levee points and IFAs
Flow data - Full discharges through Kaufman LID 15 with reduced discharges from STA 9844-16998 based on With Levee supplemental model that used lateral structure to represent spill to the Trinity River

--- EF_FEMA.p06 (plan) ---

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Plan Title=ScenarioG_EastFork_Kauf_MUD1_NV_FW
Short Identifier=ScenarioG_FW
Geom File=g01
Flow File=f06
Encroach River=East Fork
Encroach Reach=1
Encroach Node=39720
       110984.68   13640
Encroach Node=38555
       1   10565   13815
Encroach Node=37574
       1   10820   14910
Encroach Node=36633
       1    9561   14325
Encroach Node=35477
       1    8052   13625
Encroach Node=34584
       1    6222   12525
Encroach Node=33667
       1    4788   12025
Encroach Node=32592
       1    7500   15175
Encroach Node=31621
       1    6450   14650
Encroach Node=30803
       1    6350   14600
Encroach Node=29740
       1    9860   17800
Encroach Node=28442
       1    9825   17480
Encroach Node=27695
       1    8800   16050
Encroach Node=26944
       1   12450   19400
Encroach Node=26212
       1   12800   19750
Encroach Node=25584
       1   12700   19580
Encroach Node=24832
       1   12800   19900
Encroach Node=23467
       1   12300   19700
Encroach Node=22521
       1   12000   19510
Encroach Node=21721
       1   11700   19400
Encroach Node=21095
       1   1140019458.57
Encroach Node=20992
       1    7000   15525
Encroach Node=20892
       1   1100019609.65
Encroach Node=19745
       1   1080019919.55
Encroach Node=18741
       1   11900   20950
Encroach Node=16998
       1   12500   21350
Encroach Node=16194
       1   12700   21250
Encroach Node=14669
       1   12850   20955
Encroach Node=12629
       1   1290020800.67
Encroach Node=11232
       1   1280020356.08
Encroach Node=9844
       1   12750   19670

--- EF_FEMA.p07 (plan) ---

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Plan Title=ScenarioH_EastFork_Kauf_5_East_NV_FW
Short Identifier=ScenarioH_FW
Geom File=g02
Flow File=f04
Encroach River=East Fork
Encroach Reach=1
Encroach Node=53041
       1    2725 9116.72
Encroach Node=52589
       1    2575 9010.77
Encroach Node=51649
       1    2650 8952.03
Encroach Node=50644
       1    2800 9051.15
Encroach Node=49796
       1    2975 9037.38
Encroach Node=48320
       1    3300 8886.59
Encroach Node=47200
       1    3600 9075.86
Encroach Node=46345
       1    3950 9373.59
Encroach Node=45584
       1    4400   10350
Encroach Node=44251
       1    2500    7700
Encroach Node=42906
       1    3900    8650
Encroach Node=42075
       1    5500    9850
Encroach Node=40855
       1    5300    9275
Encroach Node=39720
       110950.43   13640
Encroach Node=38555
       1 11428.5   13815
Encroach Node=37574
       1 12409.1   14910
Encroach Node=36633
       112226.18   14325
Encroach Node=35477
       112272.22   13625
Encroach Node=34584
       111175.22   12525
Encroach Node=33667
       1 10426.8   12025
Encroach Node=32592
       113572.15   15175
Encroach Node=31621
       113021.42   14650
Encroach Node=30803
       113062.08   14600
Encroach Node=29740
       116246.72   17800
Encroach Node=28442
       115974.51   17480
Encroach Node=27695
       114533.59   16050
Encroach Node=26944
       117898.69   19400
Encroach Node=26212
       118199.59   19750
Encroach Node=25584
       118107.54   19580
Encroach Node=24832
       118457.09   19900
Encroach Node=23467
       118342.04   19700
Encroach Node=22521
       118144.05   19510
Encroach Node=21721
       118021.93   19400
Encroach Node=21095
       1 17954.619458.57
Encroach Node=20992
       113827.64   15525
Encroach Node=20892
       117893.2419609.65
Encroach Node=19745
       117696.5119919.55
Encroach Node=18741
       118773.96   20950
Encroach Node=16998
       119522.83   21350
Encroach Node=16194
       119490.59   21250
Encroach Node=14669
       119267.92   20955
Encroach Node=12629
       119091.3420800.67
Encroach Node=11232
       118361.8620356.08
Encroach Node=9844
       118007.47   19670

--- EF_FEMA.p08 (plan) ---

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Plan Title=ScenarioI_EastFork_Kauf_5_West_NV_FW
Short Identifier=ScenarioI_FW
Geom File=g03
Flow File=f04
Encroach River=East Fork
Encroach Reach=1
Encroach Node=53041
       1 3127.82    9095
Encroach Node=52589
       1 6041.69    9000
Encroach Node=51649
       1 7343.68   10200
Encroach Node=50644
       1 7726.22   12643
Encroach Node=49796
       1 7658.58   13300
Encroach Node=48320
       1 7328.48   12104
Encroach Node=47200
       1 7698.34   10693
Encroach Node=46345
       1    8018   10250
Encroach Node=45584
       1    8533   10350
Encroach Node=44251
       1 5514.81    7700
Encroach Node=42906
       1 6994.35    8650
Encroach Node=42075
       1 8028.37    9850
Encroach Node=40855
       1 7360.37    9275
Encroach Node=39720
       110950.43   13640
Encroach Node=38555
       1 11428.5   13815
Encroach Node=37574
       1 12409.1   14910
Encroach Node=36633
       112226.18   14325
Encroach Node=35477
       112272.22   13625
Encroach Node=34584
       111175.22   12525
Encroach Node=33667
       1 10426.8   12025
Encroach Node=32592
       113572.15   15175
Encroach Node=31621
       113021.42   14650
Encroach Node=30803
       113062.08   14600
Encroach Node=29740
       116246.72   17800
Encroach Node=28442
       115974.51   17480
Encroach Node=27695
       114533.59   16050
Encroach Node=26944
       117898.69   19400
Encroach Node=26212
       118199.59   19750
Encroach Node=25584
       118107.54   19580
Encroach Node=24832
       118457.09   19900
Encroach Node=23467
       118342.04   19700
Encroach Node=22521
       118144.05   19510
Encroach Node=21721
       118021.93   19400
Encroach Node=21095
       1 17954.619458.57
Encroach Node=20992
       113827.64   15525
Encroach Node=20892
       117893.2419609.65
Encroach Node=19745
       117696.5119919.55
Encroach Node=18741
       118773.96   20950
Encroach Node=16998
       119522.83   21350
Encroach Node=16194
       119490.59   21250
Encroach Node=14669
       119267.92   20955
Encroach Node=12629
       119091.3420800.67
Encroach Node=11232
       118361.8620356.08
Encroach Node=9844
       118007.47   19670

--- EF_FEMA.p09 (plan) ---

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Plan Title=ScenarioJ_EastFork_Kauf_LID10_NV_FW
Short Identifier=ScenarioJ_FW
Geom File=g04
Flow File=f04
Encroach River=East Fork
Encroach Reach=1
Encroach Node=66590
       1    4000    9450
Encroach Node=64748
       1    2200    8225
Encroach Node=63490
       1    2400    8100
Encroach Node=62827
       1    2600    8025
Encroach Node=62107
       1    3950    9000
Encroach Node=61773
       1    3720    8695
Encroach Node=61239
       1    3715    8650
Encroach Node=61008
       1    3530    8675
Encroach Node=59796
       1    3550    8400
Encroach Node=58768
       1    3810    7850
Encroach Node=57547
       1    4075    7575
Encroach Node=56456
       1    3890    7575
Encroach Node=54807
       1    3680    8075
Encroach Node=54191
       1    3640 8898.11
Encroach Node=53843
       1    3600 9348.54
Encroach Node=53041
       1 3127.82 9116.72
Encroach Node=52589
       1 6041.69 9010.77
Encroach Node=51649
       1 7343.68 8952.03
Encroach Node=50644
       1 7726.22 9051.15
Encroach Node=49796
       1 7658.58 9037.38
Encroach Node=48320
       1 7328.48 8886.59
Encroach Node=47200
       1 7698.34 9075.86
Encroach Node=46345
       1    8018 9373.59
Encroach Node=45584
       1    8533   10350
Encroach Node=44251
       1 5514.81    7700
Encroach Node=42906
       1 6994.35    8650
Encroach Node=42075
       1 8028.37    9850
Encroach Node=40855
       1 7360.37    9275
Encroach Node=39720
       110950.43   13640
Encroach Node=38555
       1 11428.5   13815
Encroach Node=37574
       1 12409.1   14910
Encroach Node=36633
       112226.18   14325
Encroach Node=35477
       112272.22   13625
Encroach Node=34584
       111175.22   12525
Encroach Node=33667
       1 10426.8   12025
Encroach Node=32592
       113572.15   15175
Encroach Node=31621
       113021.42   14650
Encroach Node=30803
       113062.08   14600
Encroach Node=29740
       116246.72   17800
Encroach Node=28442
       115974.51   17480
Encroach Node=27695
       114533.59   16050
Encroach Node=26944
       117898.69   19400
Encroach Node=26212
       118199.59   19750
Encroach Node=25584
       118107.54   19580
Encroach Node=24832
       118457.09   19900
Encroach Node=23467
       118342.04   19700
Encroach Node=22521
       118144.05   19510
Encroach Node=21721
       118021.93   19400
Encroach Node=21095
       1 17954.619458.57
Encroach Node=20992
       113827.64   15525
Encroach Node=20892
       117893.2419609.65
Encroach Node=19745
       117696.5119919.55
Encroach Node=18741
       118773.96   20950
Encroach Node=16998
       119522.83   21350
Encroach Node=16194
       119490.59   21250
Encroach Node=14669
       119267.92   20955
Encroach Node=12629
       119091.3420800.67
Encroach Node=11232
       118361.8620356.08
Encroach Node=9844
       118007.47   19670

--- EF_FEMA.p10 (plan) ---

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Plan Title=ScenarioK_EastFork_Kauf_LID15_NV_FW
Short Identifier=ScenarioK_FW
Geom File=g05
Flow File=f02
Encroach River=East Fork
Encroach Reach=1
Encroach Node=94766
       1    5726    9000
Encroach Node=93866
       1 7123.13    9950
Encroach Node=91923
       1    6500   10100
Encroach Node=90416
       1    7500   13000
Encroach Node=89281
       1    7475   13250
Encroach Node=88315
       1    7775   13400
Encroach Node=86331
       1    7350   12725
Encroach Node=85652
       1 6639.68   12350
Encroach Node=84705
       1    5600   12150
Encroach Node=83642
       1    4139   12826
Encroach Node=83532
       1    3900   12784
Encroach Node=82836
       1    3350   12300
Encroach Node=81963
       1    2650   11471
Encroach Node=81004
       1    2600   11350
Encroach Node=77836
       1    2100   10700
Encroach Node=77092
       1    2100   10250
Encroach Node=75815
       1    2050    9100
Encroach Node=74927
       1    2000 8421.44
Encroach Node=72977
       1    1850    7725
Encroach Node=72378
       1    2500    8450
Encroach Node=70658
       1    3800    9950
Encroach Node=68622
       1    5650   11450
Encroach Node=66590
       1    4000 8094.32
Encroach Node=64748
       1    2200 6047.81
Encroach Node=63490
       1    2400 5882.69
Encroach Node=62827
       1    2600 6090.88
Encroach Node=62107
       1    3950 7061.51
Encroach Node=61773
       1    3720 6652.11
Encroach Node=61239
       1    3715 6812.19
Encroach Node=61008
       1    3530 6700.57
Encroach Node=59796
       1    3550 6650.54
Encroach Node=58768
       1    3810 6838.77
Encroach Node=57547
       1    4075 6662.86
Encroach Node=56456
       1    3890  6753.8
Encroach Node=54807
       1    3680 7620.06
Encroach Node=54191
       1    3640 8898.11
Encroach Node=53843
       1    3600 9348.54
Encroach Node=53041
       1 3127.82 9116.72
Encroach Node=52589
       1 6041.69 9010.77
Encroach Node=51649
       1 7343.68 8952.03
Encroach Node=50644
       1 7726.22 9051.15
Encroach Node=49796
       1 7658.58 9037.38
Encroach Node=48320
       1 7328.48 8886.59
Encroach Node=47200
       1 7698.34 9075.86
Encroach Node=46345
       1    8018 9373.59
Encroach Node=45584
       1    8533   10350
Encroach Node=44251
       1 5514.81    7700
Encroach Node=42906
       1 6994.35    8650
Encroach Node=42075
       1 8028.37    9850
Encroach Node=40855
       1 7360.37    9275
Encroach Node=39720
       110950.43   13640
Encroach Node=38555
       1 11428.5   13815
Encroach Node=37574
       1 12409.1   14910
Encroach Node=36633
       112226.18   14325
Encroach Node=35477
       112272.22   13625
Encroach Node=34584
       111175.22   12525
Encroach Node=33667
       1 10426.8   12025
Encroach Node=32592
       113572.15   15175
Encroach Node=31621
       113021.42   14650
Encroach Node=30803
       113062.08   14600
Encroach Node=29740
       116246.72   17800
Encroach Node=28442
       115974.51   17480
Encroach Node=27695
       114533.59   16050
Encroach Node=26944
       117898.69   19400
Encroach Node=26212
       118199.59   19750
Encroach Node=25584
       118107.54   19580
Encroach Node=24832
       118457.09   19900
Encroach Node=23467
       118342.04   19700
Encroach Node=22521
       118144.05   19510
Encroach Node=21721
       118021.93   19400
Encroach Node=21095
       1 17954.619458.57
Encroach Node=20992
       113827.64   15525
Encroach Node=20892
       117893.2419609.65
Encroach Node=19745
       117696.5119919.55
Encroach Node=18741
       118773.96   20950
Encroach Node=16998
       119522.83   21350
Encroach Node=16194
       119490.59   21250
Encroach Node=14669
       119267.92   20955
Encroach Node=12629
       119091.3420800.67
Encroach Node=11232
       118361.8620356.08
Encroach Node=9844
       118007.47   19670

--- EF_FEMA.p12 (plan) ---

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Plan Title=EastFork_WithLevee_FW
Short Identifier=WithLevee_FW
Geom File=g06
Flow File=f04
Encroach River=East Fork
Encroach Reach=1
Encroach Node=154701
       1  642.09    8230
Encroach Node=153755
       1  665.86    4390
Encroach Node=152745
       1    1885    6500
Encroach Node=151671
       1    2305    8395
Encroach Node=150670
       1    3505   10065
Encroach Node=149657
       1    4200   11420
Encroach Node=148653
       1    4180   11970
Encroach Node=147648
       1    1380    9135
Encroach Node=146847
       1     795    8195
Encroach Node=145933
       1  603.71 6479.85
Encroach Node=145581
       1     800  6670.4
Encroach Node=144984
       1  633.54    7230
Encroach Node=144246
       1  822.25    7605
Encroach Node=141955
       1 1426.16    8200
Encroach Node=140162
       1    1450    8560
Encroach Node=137347
       1    5030   11860
Encroach Node=135946
       1    5440   11750
Encroach Node=134267
       1    5305   11680
Encroach Node=133019
       1    5220   11900
Encroach Node=131615
       1    462512215.42
Encroach Node=131320
       1    4590   12115
Encroach Node=131178
       1    452511862.26
Encroach Node=130522
       1    3198 9288.19
Encroach Node=129244
       1    3100  9702.9
Encroach Node=128203
       1    3020  8586.9
Encroach Node=127187
       1    2915  8456.7
Encroach Node=126440
       1    2480  7321.2
Encroach Node=125131
       1    3090  8280.3
Encroach Node=124014
       1    2950    8700
Encroach Node=123188
       1    1950    8000
Encroach Node=122311
       1    1090    7350
Encroach Node=120494
       1    1550    8000
Encroach Node=118625
       1    3430    9800
Encroach Node=115837
       1    2600  9529.2
Encroach Node=114150
       1    2250 10120.2
Encroach Node=112120
       1    3450 11345.4
Encroach Node=111013
       1    4500   10735
Encroach Node=108510
       1    5400   10800
Encroach Node=107423
       1    3760    9280
Encroach Node=106628
       1    3640    9200
Encroach Node=105627
       1    3590    9360
Encroach Node=104782
       1    3480    9930
Encroach Node=103602
       1    3450   10865
Encroach Node=102905
       1    3450   11250
Encroach Node=102352
       1    3100   10900
Encroach Node=101670
       1    3150   10900
Encroach Node=100387
       1    3200   10550
Encroach Node=97061
       1    3800   10100
Encroach Node=96048
       1    4227    9400
Encroach Node=94766
       1    5726    9000
Encroach Node=93866
       1 7123.13    9950
Encroach Node=91923
       1 7977.49   10100
Encroach Node=90416
       110059.86   13000
Encroach Node=89281
       1 10686.1   13250
Encroach Node=88315
       111297.45   13400
Encroach Node=86331
       111216.57   12725
Encroach Node=85652
       110900.99   12350
Encroach Node=84705
       1 10761.9   12150
Encroach Node=83642
       110533.18   12826
Encroach Node=83532
       110484.75   12784
Encroach Node=82836
       110281.69   12300
Encroach Node=81963
       1 9351.78   11471
Encroach Node=81004
       1 8248.64   11350
Encroach Node=77836
       1 7746.53   10700
Encroach Node=77092
       1 7731.38   10250
Encroach Node=75815
       1 7616.06    9100
Encroach Node=74927
       1 7047.42 8421.44
Encroach Node=72977
       1 6008.65    7725
Encroach Node=72378
       1 6402.85    8450
Encroach Node=70658
       1  7185.4    9950
Encroach Node=68622
       1    5650   11450
Encroach Node=66590
       1    4000 8094.32
Encroach Node=64748
       1    2200 6047.81
Encroach Node=63490
       1    2400 5882.69
Encroach Node=62827
       1    2600 6090.88
Encroach Node=62107
       1    3950 7061.51
Encroach Node=61773
       1    3720 6652.11
Encroach Node=61239
       1    3715 6812.19
Encroach Node=61008
       1    3530 6700.57
Encroach Node=59796
       1    3550 6650.54
Encroach Node=58768
       1    3810 6838.77
Encroach Node=57547
       1    4075 6662.86
Encroach Node=56456
       1    3890  6753.8
Encroach Node=54807
       1    3680 7620.06
Encroach Node=54191
       1    3640 8898.11
Encroach Node=53843
       1    3600 9348.54
Encroach Node=53041
       1 3127.82 9116.72
Encroach Node=52589
       1 6041.69 9010.77
Encroach Node=51649
       1 7343.68 8952.03
Encroach Node=50644
       1 7726.22 9051.15
Encroach Node=49796
       1 7658.58 9037.38
Encroach Node=48320
       1 7328.48 8886.59
Encroach Node=47200
       1 7698.34 9075.86
Encroach Node=46345
       1    8018 9373.59
Encroach Node=45584
       1    8533   10350
Encroach Node=44251
       1 5514.81    7700
Encroach Node=42906
       1 6994.35    8650
Encroach Node=42075
       1 8028.37    9850
Encroach Node=40855
       1 7360.37    9275
Encroach Node=39720
       110950.43   13640
Encroach Node=38555
       1 11428.5   13815
Encroach Node=37574
       1 12409.1   14910
Encroach Node=36633
       112226.18   14325
Encroach Node=35477
       112272.22   13625
Encroach Node=34584
       111175.22   12525
Encroach Node=33667
       1 10426.8   12025
Encroach Node=32592
       113572.15   15175
Encroach Node=31621
       113021.42   14650
Encroach Node=30803
       113062.08   14600
Encroach Node=29740
       116246.72   17800
Encroach Node=28442
       115974.51   17480
Encroach Node=27695
       114533.59   16050
Encroach Node=26944
       117898.69   19400
Encroach Node=26212
       118199.59   19750
Encroach Node=25584
       118107.54   19580
Encroach Node=24832
       118457.09   19900
Encroach Node=23467
       118342.04   19700
Encroach Node=22521
       118144.05   19510
Encroach Node=21721
       118021.93   19400
Encroach Node=21095
       1 17954.619458.57
Encroach Node=20992
       113827.64   15525
Encroach Node=20892
       117893.2419609.65
Encroach Node=19745
       117696.5119919.55
Encroach Node=18741
       118773.96   20950
Encroach Node=16998
       119522.83   21350
Encroach Node=16194
       119490.59   21250
Encroach Node=14669
       119267.92   20955
Encroach Node=12629
       119091.3420800.67
Encroach Node=11232
       118361.8620356.08
Encroach Node=9844
       118007.47   19670

--- EF_FEMA.f03 (steady flow) ---

Flow Title=2020 Reduced East Fork Discharges
Program Version=5.06
BEGIN FILE DESCRIPTION:
Reduced discharges through Kaufman LID 15 based on With Levee supplemental model that used a lateral structure to represent the levee and from STA 9844-16998 based on With Levee supplemental model that used lateral structure to represent spill to the Trinity River with full discharges elsewhere.
Boundary condition - Normal depth slope=0.0003 based on East Fork survey data
END FILE DESCRIPTION:
Number of Profiles= 7
Profile Names=10YR,25YR,50YR,100YR,500YR,1PCT_MINUS,1PCT_PLUS
River Rch & RM=East Fork,1               ,154701
   26000   38000   47400   59800  101300   39700  108900
River Rch & RM=East Fork,1               ,148653
   30300   44100   55000   69300  117100   46200  125300
River Rch & RM=East Fork,1               ,135946
   28300   42900   55800   71900  123600   48000  130600
River Rch & RM=East Fork,1               ,111013
   25200   37500   50300   67000  117600   43300  127300
River Rch & RM=East Fork,1               ,94766
   25200   37500   50300   67000  114015   43300  122506
River Rch & RM=East Fork,1               ,93866
   25200   37500   50299   66790  107903   43300  114692
River Rch & RM=East Fork,1               ,91923
   25200   37500   50110   64455   96554   43300  102170
River Rch & RM=East Fork,1               ,90416
   25200   37475   49149   61498   87697   42991   92589
River Rch & RM=East Fork,1               ,89281
   25200   37475   48617   59038   79887   42955   84086
River Rch & RM=East Fork,1               ,88315
   25200   37475   48576   58266   75843   42955   79474
River Rch & RM=East Fork,1               ,86331
   25200   37475   48466   57238   71466   42955   74488
River Rch & RM=East Fork,1               ,85652
   25200   37475   48466   57162   70733   42955   73601
River Rch & RM=East Fork,1               ,84705
   25200   37475   48466   57152   70460   42955   73219
River Rch & RM=East Fork,1               ,83642
   25200   37475   48324   56641   69023   42934   71528
River Rch & RM=East Fork,1               ,83532
   25200   37475   48324   56641   69023   42934   71528
River Rch & RM=East Fork,1               ,82836
   25200   37475   48242   55931   66393   42927   68206
River Rch & RM=East Fork,1               ,81963
   25200   37475   48198   55478   64226   42926   65232
River Rch & RM=East Fork,1               ,81004
   25200   37475   48159   54776   60196   42926   59346
River Rch & RM=East Fork,1               ,77836
   25200   37475   48159   54770   59678   42926   58343
River Rch & RM=East Fork,1               ,77092
   25200   37475   48159   54770   59577   42926   57999
River Rch & RM=East Fork,1               ,75815
   25200   37475   48159   54770   58106   42926   55263
River Rch & RM=East Fork,1               ,74927
   25200   37475   48159   54714   56235   42926   52296
River Rch & RM=East Fork,1               ,72977
   25200   37475   48159   54558   47058   42926   40150
River Rch & RM=East Fork,1               ,72378
   25200   37475   48159   54550   42408   42926   35002
River Rch & RM=East Fork,1               ,70658
   25200   37475   48159   54549   36219   42926   28046
River Rch & RM=East Fork,1               ,68622
   23500   33175   42159   45949   16919   38626    6746
River Rch & RM=East Fork,1               ,66590
   23500   33200   44300   58400   98300   39000  106000
River Rch & RM=East Fork,1               ,23467
   20600   28700   37100   48600   75100   33700   83400
River Rch & RM=East Fork,1               ,16998
   20600   28641   36245   45558   64151   33256   69658
River Rch & RM=East Fork,1               ,16194
   20600   28641   36245   45558   63128   33256   67839
River Rch & RM=East Fork,1               ,14669
   20600   28641   36245   45558   62882   33256   66945
River Rch & RM=East Fork,1               ,12629
   20600   28641   36245   45558   62857   33256   66878
River Rch & RM=East Fork,1               ,11232
   20600   28641   36245   45558   62857   33256   66878
River Rch & RM=East Fork,1               ,9844
   20600   28641   36245   45558   62857   33256   66878
Boundary for River Rch & Prof#=East Fork,1               , 1
Up Type= 0
Dn Type= 3
Dn Slope=0.0003
Boundary for River Rch & Prof#=East Fork,1               , 2
Up Type= 0
Dn Type= 3
Dn Slope=0.0003
Boundary for River Rch & Prof#=East Fork,1               , 3
Up Type= 0
Dn Type= 3
Dn Slope=0.0003
Boundary for River Rch & Prof#=East Fork,1               , 4
Up Type= 0
Dn Type= 3
Dn Slope=0.0003
Boundary for River Rch & Prof#=East Fork,1               , 5
Up Type= 0
Dn Type= 3
Dn Slope=0.0003
Boundary for River Rch & Prof#=East Fork,1               , 6
Up Type= 0
Dn Type= 3
Dn Slope=0.0003
Boundary for River Rch & Prof#=East Fork,1               , 7
Up Type= 0
Dn Type= 3
Dn Slope=0.0003
Initial Flow Split=East Fork       ,12030106000003  ,96047   ,
       0   23.87  2544.813820.26   60000       0       0
Initial Flow Split=East Fork       ,12030106000003  ,18740   ,
       0       0  317.76 2354.05 10786.6       0       0
DSS Import GetInterval= 0
DSS Import GetPeak= 0
DSS Import FillOption= 0

--- EF_FEMA.f01 (steady flow) ---

Flow Title=2020 Kaufman LID15 Reduced Discharges
Program Version=5.06
BEGIN FILE DESCRIPTION:
Full discharges through Kaufman LID 15 with reduced discharges from STA 9844-16998 based on With Levee supplemental model that used lateral structure to represent spill to the Trinity River
Boundary condition - Normal depth slope=0.0003 based on East Fork survey data
END FILE DESCRIPTION:
Number of Profiles= 7
Profile Names=10YR,25YR,50YR,100YR,500YR,1PCT_MINUS,1PCT_PLUS
River Rch & RM=East Fork,1               ,154701
   26000   38000   47400   59800  101300   39700  108900
River Rch & RM=East Fork,1               ,148653
   30300   44100   55000   69300  117100   46200  125300
River Rch & RM=East Fork,1               ,135946
   28300   42900   55800   71900  123600   48000  130600
River Rch & RM=East Fork,1               ,111013
   25200   37500   50300   67000  117600   43300  127300
River Rch & RM=East Fork,1               ,68622
   23500   33200   44300   58400   98300   39000  106000
River Rch & RM=East Fork,1               ,23467
   20600   28700   37100   48600   75100   33700   83400
River Rch & RM=East Fork,1               ,16998
   20600   28641   36245   45558   64151   33256   69658
River Rch & RM=East Fork,1               ,16194
   20600   28641   36245   45558   63128   33256   67839
River Rch & RM=East Fork,1               ,14669
   20600   28641   36245   45558   62882   33256   66945
River Rch & RM=East Fork,1               ,12629
   20600   28641   36245   45558   62857   33256   66878
River Rch & RM=East Fork,1               ,11232
   20600   28641   36245   45558   62857   33256   66878
River Rch & RM=East Fork,1               ,9844
   20600   28641   36245   45558   62857   33256   66878
Boundary for River Rch & Prof#=East Fork,1               , 1
Up Type= 0
Dn Type= 3
Dn Slope=0.0003
Boundary for River Rch & Prof#=East Fork,1               , 2
Up Type= 0
Dn Type= 3
Dn Slope=0.0003
Boundary for River Rch & Prof#=East Fork,1               , 3
Up Type= 0
Dn Type= 3
Dn Slope=0.0003
Boundary for River Rch & Prof#=East Fork,1               , 4
Up Type= 0
Dn Type= 3
Dn Slope=0.0003
Boundary for River Rch & Prof#=East Fork,1               , 5
Up Type= 0
Dn Type= 3
Dn Slope=0.0003
Boundary for River Rch & Prof#=East Fork,1               , 6
Up Type= 0
Dn Type= 3
Dn Slope=0.0003
Boundary for River Rch & Prof#=East Fork,1               , 7
Up Type= 0
Dn Type= 3
Dn Slope=0.0003
Initial Flow Split=East Fork       ,12030106000003  ,96047   ,
       0   23.87  2544.813820.26   60000       0       0
Initial Flow Split=East Fork       ,12030106000003  ,18740   ,
       0       0  317.76 2354.05 10786.6       0       0
DSS Import GetInterval= 0
DSS Import GetPeak= 0
DSS Import FillOption= 0

--- EF_FEMA.f02 (steady flow) ---

Flow Title=2020 Kaufman LID15 Reduced Discharges_FW
Program Version=5.06
Number of Profiles= 2
Profile Names=100YR,FW
River Rch & RM=East Fork,1               ,154701
   59800   59800
River Rch & RM=East Fork,1               ,148653
   69300   69300
River Rch & RM=East Fork,1               ,135946
   71900   71900
River Rch & RM=East Fork,1               ,111013
   67000   67000
River Rch & RM=East Fork,1               ,68622
   58400   58400
River Rch & RM=East Fork,1               ,23467
   48600   48600
River Rch & RM=East Fork,1               ,16998
   45558   45558
Boundary for River Rch & Prof#=East Fork,1               , 1
Up Type= 0
Dn Type= 3
Dn Slope=0.0003
Boundary for River Rch & Prof#=East Fork,1               , 2
Up Type= 0
Dn Type= 3
Dn Slope=0.0003
Initial Flow Split=East Fork       ,12030106000003  ,96047   ,
       0   23.87
Initial Flow Split=East Fork       ,12030106000003  ,18740   ,
       0       0
DSS Import GetInterval= 0
DSS Import GetPeak= 0
DSS Import FillOption= 0

--- EF_FEMA.f04 (steady flow) ---

Flow Title=2020 Reduced East Fork Discharges_FW
Program Version=5.06
Number of Profiles= 2
Profile Names=100YR,FW
River Rch & RM=East Fork,1               ,154701
   59800   59800
River Rch & RM=East Fork,1               ,148653
   69300   69300
River Rch & RM=East Fork,1               ,135946
   71900   71900
River Rch & RM=East Fork,1               ,111013
   67000   67000
River Rch & RM=East Fork,1               ,94766
   67000   67000
River Rch & RM=East Fork,1               ,93866
   66790   66790
River Rch & RM=East Fork,1               ,91923
   64455   64455
River Rch & RM=East Fork,1               ,90416
   61498   61498
River Rch & RM=East Fork,1               ,89281
   59038   59038
River Rch & RM=East Fork,1               ,88315
   58266   58266
River Rch & RM=East Fork,1               ,86331
   57238   57238
River Rch & RM=East Fork,1               ,85652
   57162   57162
River Rch & RM=East Fork,1               ,84705
   57152   57152
River Rch & RM=East Fork,1               ,83642
   56641   56641
River Rch & RM=East Fork,1               ,83532
   56641   56641
River Rch & RM=East Fork,1               ,82836
   55931   55931
River Rch & RM=East Fork,1               ,81963
   55478   55478
River Rch & RM=East Fork,1               ,81004
   54776   54776
River Rch & RM=East Fork,1               ,77836
   54770   54770
River Rch & RM=East Fork,1               ,77092
   54770   54770
River Rch & RM=East Fork,1               ,75815
   54770   54770
River Rch & RM=East Fork,1               ,74927
   54714   54714
River Rch & RM=East Fork,1               ,72977
   54558   54558
River Rch & RM=East Fork,1               ,72378
   54550   54550
River Rch & RM=East Fork,1               ,70658
   54549   54549
River Rch & RM=East Fork,1               ,68622
   45949   45949
River Rch & RM=East Fork,1               ,66590
   58400   58400
River Rch & RM=East Fork,1               ,23467
   48600   48600
River Rch & RM=East Fork,1               ,16998
   45558   45558
Boundary for River Rch & Prof#=East Fork,1               , 1
Up Type= 0
Dn Type= 3
Dn Slope=0.0003
Boundary for River Rch & Prof#=East Fork,1               , 2
Up Type= 0
Dn Type= 3
Dn Slope=0.0003
Initial Flow Split=East Fork       ,12030106000003  ,96047   ,
       0   23.87
Initial Flow Split=East Fork       ,12030106000003  ,18740   ,
       0       0
DSS Import GetInterval= 0
DSS Import GetPeak= 0
DSS Import FillOption= 0

--- EF_FEMA.f05 (steady flow) ---

Flow Title=2020 Kaufman MUD1 Reduced Discharges
Program Version=5.06
BEGIN FILE DESCRIPTION:
Full discharges through Kaufman MUD 1 with reduced discharges through Kaufman LID 15 based on With Levee supplemental model that used a lateral structure to represent the levee
Boundary condition - Normal depth slope=0.0003 based on East Fork survey data
END FILE DESCRIPTION:
Number of Profiles= 7
Profile Names=10YR,25YR,50YR,100YR,500YR,1PCT_MINUS,1PCT_PLUS
River Rch & RM=East Fork,1               ,154701
   26000   38000   47400   59800  101300   39700  108900
River Rch & RM=East Fork,1               ,148653
   30300   44100   55000   69300  117100   46200  125300
River Rch & RM=East Fork,1               ,135946
   28300   42900   55800   71900  123600   48000  130600
River Rch & RM=East Fork,1               ,111013
   25200   37500   50300   67000  117600   43300  127300
River Rch & RM=East Fork,1               ,94766
   25200   37500   50300   67000  114015   43300  122506
River Rch & RM=East Fork,1               ,93866
   25200   37500   50299   66790  107903   43300  114692
River Rch & RM=East Fork,1               ,91923
   25200   37500   50110   64455   96554   43300  102170
River Rch & RM=East Fork,1               ,90416
   25200   37475   49149   61498   87697   42991   92589
River Rch & RM=East Fork,1               ,89281
   25200   37475   48617   59038   79887   42955   84086
River Rch & RM=East Fork,1               ,88315
   25200   37475   48576   58266   75843   42955   79474
River Rch & RM=East Fork,1               ,86331
   25200   37475   48466   57238   71466   42955   74488
River Rch & RM=East Fork,1               ,85652
   25200   37475   48466   57162   70733   42955   73601
River Rch & RM=East Fork,1               ,84705
   25200   37475   48466   57152   70460   42955   73219
River Rch & RM=East Fork,1               ,83642
   25200   37475   48324   56641   69023   42934   71528
River Rch & RM=East Fork,1               ,83532
   25200   37475   48324   56641   69023   42934   71528
River Rch & RM=East Fork,1               ,82836
   25200   37475   48242   55931   66393   42927   68206
River Rch & RM=East Fork,1               ,81963
   25200   37475   48198   55478   64226   42926   65232
River Rch & RM=East Fork,1               ,81004
   25200   37475   48159   54776   60196   42926   59346
River Rch & RM=East Fork,1               ,77836
   25200   37475   48159   54770   59678   42926   58343
River Rch & RM=East Fork,1               ,77092
   25200   37475   48159   54770   59577   42926   57999
River Rch & RM=East Fork,1               ,75815
   25200   37475   48159   54770   58106   42926   55263
River Rch & RM=East Fork,1               ,74927
   25200   37475   48159   54714   56235   42926   52296
River Rch & RM=East Fork,1               ,72977
   25200   37475   48159   54558   47058   42926   40150
River Rch & RM=East Fork,1               ,72378
   25200   37475   48159   54550   42408   42926   35002
River Rch & RM=East Fork,1               ,70658
   25200   37475   48159   54549   36219   42926   28046
River Rch & RM=East Fork,1               ,68622
   23500   33175   42159   45949   16919   38626    6746
River Rch & RM=East Fork,1               ,66590
   23500   33200   44300   58400   98300   39000  106000
River Rch & RM=East Fork,1               ,23467
   20600   28700   37100   48600   75100   33700   83400
Boundary for River Rch & Prof#=East Fork,1               , 1
Up Type= 0
Dn Type= 3
Dn Slope=0.0003
Boundary for River Rch & Prof#=East Fork,1               , 2
Up Type= 0
Dn Type= 3
Dn Slope=0.0003
Boundary for River Rch & Prof#=East Fork,1               , 3
Up Type= 0
Dn Type= 3
Dn Slope=0.0003
Boundary for River Rch & Prof#=East Fork,1               , 4
Up Type= 0
Dn Type= 3
Dn Slope=0.0003
Boundary for River Rch & Prof#=East Fork,1               , 5
Up Type= 0
Dn Type= 3
Dn Slope=0.0003
Boundary for River Rch & Prof#=East Fork,1               , 6
Up Type= 0
Dn Type= 3
Dn Slope=0.0003
Boundary for River Rch & Prof#=East Fork,1               , 7
Up Type= 0
Dn Type= 3
Dn Slope=0.0003
Initial Flow Split=East Fork       ,12030106000003  ,96047   ,
       0   23.87  2544.813820.26   60000       0       0
Initial Flow Split=East Fork       ,12030106000003  ,18740   ,
       0       0  317.76 2354.05 10786.6       0       0
DSS Import GetInterval= 0
DSS Import GetPeak= 0
DSS Import FillOption= 0

--- EF_FEMA.f06 (steady flow) ---

Flow Title=2020 Kaufman MUD1 Reduced Discharges_FW
Program Version=5.06
Number of Profiles= 2
Profile Names=100YR,FW
River Rch & RM=East Fork,1               ,154701
   59800   59800
River Rch & RM=East Fork,1               ,148653
   69300   69300
River Rch & RM=East Fork,1               ,135946
   71900   71900
River Rch & RM=East Fork,1               ,111013
   67000   67000
River Rch & RM=East Fork,1               ,94766
   67000   67000
River Rch & RM=East Fork,1               ,93866
   66790   66790
River Rch & RM=East Fork,1               ,91923
   64455   64455
River Rch & RM=East Fork,1               ,90416
   61498   61498
River Rch & RM=East Fork,1               ,89281
   59038   59038
River Rch & RM=East Fork,1               ,88315
   58266   58266
River Rch & RM=East Fork,1               ,86331
   57238   57238
River Rch & RM=East Fork,1               ,85652
   57162   57162
River Rch & RM=East Fork,1               ,84705
   57152   57152
River Rch & RM=East Fork,1               ,83642
   56641   56641
River Rch & RM=East Fork,1               ,83532
   56641   56641
River Rch & RM=East Fork,1               ,82836
   55931   55931
River Rch & RM=East Fork,1               ,81963
   55478   55478
River Rch & RM=East Fork,1               ,81004
   54776   54776
River Rch & RM=East Fork,1               ,77836
   54770   54770
River Rch & RM=East Fork,1               ,77092
   54770   54770
River Rch & RM=East Fork,1               ,75815
   54770   54770
River Rch & RM=East Fork,1               ,74927
   54714   54714
River Rch & RM=East Fork,1               ,72977
   54558   54558
River Rch & RM=East Fork,1               ,72378
   54550   54550
River Rch & RM=East Fork,1               ,70658
   54549   54549
River Rch & RM=East Fork,1               ,68622
   45949   45949
River Rch & RM=East Fork,1               ,66590
   58400   58400
River Rch & RM=East Fork,1               ,23467
   48600   48600
Boundary for River Rch & Prof#=East Fork,1               , 1
Up Type= 0
Dn Type= 3
Dn Slope=0.0003
Boundary for River Rch & Prof#=East Fork,1               , 2
Up Type= 0
Dn Type= 3
Dn Slope=0.0003
Initial Flow Split=East Fork       ,12030106000003  ,96047   ,
       0   23.87
Initial Flow Split=East Fork       ,12030106000003  ,18740   ,
       0       0
DSS Import GetInterval= 0
DSS Import GetPeak= 0
DSS Import FillOption= 0

--- EF_FEMA.f07 (steady flow) ---

Flow Title=2020 USACE East Fork Discharges
Program Version=5.06
BEGIN FILE DESCRIPTION:
-source
END FILE DESCRIPTION:
Number of Profiles= 7
Profile Names=10YR,25YR,50YR,100YR,500YR,1PCT_MINUS,1PCT_PLUS
River Rch & RM=East Fork,1               ,154701
   26000   38000   47400   59800  101300   39700  108900
River Rch & RM=East Fork,1               ,148653
   30300   44100   55000   69300  117100   46200  125300
River Rch & RM=East Fork,1               ,135946
   28300   42900   55800   71900  123600   48000  130600
River Rch & RM=East Fork,1               ,111013
   25200   37500   50300   67000  117600   43300  127300
River Rch & RM=East Fork,1               ,68622
   23500   33200   44300   58400   98300   39000  106000
River Rch & RM=East Fork,1               ,23467
   20600   28700   37100   48600   75100   33700   83400
Boundary for River Rch & Prof#=East Fork,1               , 1
Up Type= 0
Dn Type= 3
Dn Slope=0.0003
Boundary for River Rch & Prof#=East Fork,1               , 2
Up Type= 0
Dn Type= 3
Dn Slope=0.0003
Boundary for River Rch & Prof#=East Fork,1               , 3
Up Type= 0
Dn Type= 3
Dn Slope=0.0003
Boundary for River Rch & Prof#=East Fork,1               , 4
Up Type= 0
Dn Type= 3
Dn Slope=0.0003
Boundary for River Rch & Prof#=East Fork,1               , 5
Up Type= 0
Dn Type= 3
Dn Slope=0.0003
Boundary for River Rch & Prof#=East Fork,1               , 6
Up Type= 0
Dn Type= 3
Dn Slope=0.0003
Boundary for River Rch & Prof#=East Fork,1               , 7
Up Type= 0
Dn Type= 3
Dn Slope=0.0003
Initial Flow Split=East Fork       ,12030106000003  ,96047   ,
       0   23.87  2544.813820.26   60000       0       0
Initial Flow Split=East Fork       ,12030106000003  ,18740   ,
       0       0  317.76 2354.05 10786.6       0       0
DSS Import GetInterval= 0
DSS Import GetPeak= 0
DSS Import FillOption= 0

--- EF_FEMA.g06 (geometry) ---

Geom Title=EastFork_WithLevee
Program Version=5.06
BEGIN GEOM DESCRIPTION:
With Levee
END GEOM DESCRIPTION:

River Reach=East Fork       ,1
Reach XY= 30
2584433.821330736979734.484431562583285.779335476968692.78932339
2581728.704693726968715.575695142579416.421588636964977.51164898
2580529.702826636961302.381203982578265.510176556955839.46168365
2576268.982345486954556.128292312576977.315574476952473.48941298
 2575455.09355336952832.517238232576298.148953816950783.21162556
 2575204.39917286948431.128403232576390.509989566947949.18382905
2573836.343509976942249.704742482575603.70447655 6939997.9687604
2574169.676832816936589.98246615 2575233.04478486932601.26734647
 2577868.98242636928071.97030273 2578907.3937353 6928855.3906519
2580429.746333646926037.465185392584986.997061646925507.73691414
2588898.455446056923176.139543222586823.713532556910627.85525665
2588587.949833476904482.716300232590634.47756456 6902052.1607939
2593378.679425226889226.784541822590018.951892726879034.27802397
2589913.049217396875864.139023072591593.170857136873644.08703272
2590906.972754466871085.493396642584753.32692531 6869580.0679298
