--- TR_FEMA.prj (project) ---

Proj Title=Trinity_River_FEMA
Current Plan=p14
Default Exp/Contr=0.3,0.1
English Units
Geom File=g01
Geom File=g03
Geom File=g04
Geom File=g05
Geom File=g06
Geom File=g07
Geom File=g08
Flow File=f04
Flow File=f02
Flow File=f01
Flow File=f03
Flow File=f05
Flow File=f06
Flow File=f07
Flow File=f08
Flow File=f09
Flow File=f10
Flow File=f11
Flow File=f12
Flow File=f13
Flow File=f14
Flow File=f15
Plan File=p01
Plan File=p02
Plan File=p03
Plan File=p04
Plan File=p05
Plan File=p06
Plan File=p07
Plan File=p08
Plan File=p09
Plan File=p10
Plan File=p11
Plan File=p12
Plan File=p13
Plan File=p14
Background Map Layer=Levees_All
Y Axis Title=Elevation
X Axis Title(PF)=Main Channel Distance
X Axis Title(XS)=Station
BEGIN DESCRIPTION:
Trinity River Existing Conditions Steady State Model
The With Levee run contains representation of all hydraulically significant levees held in place:
Kaufman LID1/Henderson LID1 - left bank, STA 55303-downstream limit, modeled with levee points
Ellis LID2 - right bank, STA 71053-15600, modeled with levee points
Kaufman MUD 1 - left bank, STA 83616-56823
Dallas LID14/Ellis LID3 - right bank, STA 148768-80593
Bois D'Arc Levee - left bank, STA 193094-108725
Dallas LID1/Dallas LID2 - right bank, STA 204528-151264
The Natural Valley (NV) run for each levee removes representation of that levee from the model geometry while holding all other levees in place:
Scenario A - NV run of Kaufman LID1/Henderson LID1 Levee
Scenario B - NV run of Ellis LID2 Levee
Scenario C - NV run of Kaufman MUD 1 Levee
Scenario D - NV run of Dallas LID14/Ellis LID3 Levee
Scenario E - NV run of Bois D'Arc Levee
Scenario F - NV run of Dallas LID1/Dallas LID2 Levee
All field survey was based on NAVD88.
Stream Name: Trinity River
Study Extents: Southside Wastewater Treatment Plant to Henderson County
Date: April 2020
HEC-RAS v5.0.6
Prepared for: DHS/FEMA (Federal Emergency Management Agency)
Prepared by: Compass PTS JV
Contract #HSFE60-15-D-0003
Task Order #HSFE06-17-J-0047
END DESCRIPTION:
DSS File=dss
DSS Export Rating Curves= 0
DSS Export Rating Curve Sorted= 0
DSS Export Volume Flow Curves= 0
DXF Filename=C:\Users\victoria.a.nelson\Desktop\Trinity\Trinity.
DXF OffsetX= 0
DXF OffsetY= 0
DXF ScaleX= 1
DXF ScaleY= 10

--- TR_FEMA.p14 (plan) ---

Plan Title=ScenarioF_DallasLID1_DallasLID2_NV_FW
Program Version=5.06
Short Identifier=ScenarioF_FW
Geom File=g08
Flow File=f15
Subcritical Flow
K Sum by GR= 0
Std Step Tol= 0.01
Critical Tol= 0.01
Num of Std Step Trials= 20
Max Error Tol= 0.3
Flow Tol Ratio= 0.001
Split Flow NTrial= 30
Split Flow Tol= 0.02
Split Flow Ratio= 0.02
Log Output Level= 0
Friction Slope Method= 1
Unsteady Friction Slope Method= 2
Unsteady Bridges Friction Slope Method= 1
Parabolic Critical Depth
Global Vel Dist= 0 , 0 , 0
Global Log Level= 0
CheckData=True
Encroach Param=-1 ,0,0, 2
Encroach River=Trinity River
Encroach Reach=1
Encroach Node=205777
       110870.96 15599.2
Encroach Node=204528
       111531.9415770.97
Encroach Node=200569
       112186.5216387.52
Encroach Node=198513
       111895.2418718.26
Encroach Node=196991
       111797.07 20442.1
Encroach Node=195872
       1   1258821978.32
Encroach Node=194145
       113923.9225816.95
Encroach Node=193094
       113862.0626097.74
Encroach Node=191491
       115621.3526945.02
Encroach Node=189380
       117978.6529048.66
Encroach Node=187750
       118193.7929367.79
Encroach Node=186516
       120807.66   31962
Encroach Node=186264
       120792.77   31967
Encroach Node=184503
       119500.4128574.52
Encroach Node=181750
       1 17308.425306.99
Encroach Node=179572
       113460.0819660.01
Encroach Node=178698
       113289.1919079.49
Encroach Node=176021
       110296.09 17093.3
Encroach Node=172483
       113195.6319773.76
Encroach Node=169025
       114957.6723712.26
Encroach Node=167085
       116867.1925784.84
Encroach Node=165454
       1 18246.327215.59
Encroach Node=165204
       118473.1427285.44
Encroach Node=164199
       115135.9424040.38
Encroach Node=162832
       115899.0324764.83
Encroach Node=161707
       115913.2127486.73
Encroach Node=159456
       116083.7326879.97
Encroach Node=157344
       117774.12 29050.2
Encroach Node=154267
       118057.0430373.87
Encroach Node=151264
       117986.2630344.96
Encroach Node=148768
       1 16066.718258.25
Encroach Node=147333
       112596.9115036.43
Encroach Node=145717
       112408.0714387.71
Encroach Node=143893
       113381.1215611.78
Encroach Node=141890
       112814.7215382.57
Encroach Node=139225
       113073.3815128.06
Encroach Node=137179
       1 12479.5 14714.5
Encroach Node=135104
       113094.6616070.54
Encroach Node=133245
       112224.6815488.41
Encroach Node=131382
       110685.2214333.52
Encroach Node=129561
       110062.6212976.12
Encroach Node=127110
       1 9718.6112068.25
Encroach Node=124996
       1 9024.1811083.76
Encroach Node=123554
       1 8680.4711041.08
Encroach Node=122155
       1 8385.9811095.25
Encroach Node=120905
       1 8005.6910526.72
Encroach Node=118211
       1 6113.49 8803.29
Encroach Node=116211
       1  3355.6 6627.08
Encroach Node=113969
       1  3098.5 5836.82
Encroach Node=112556
       1 2584.82 5083.59
Encroach Node=110130
       1 2078.42 4345.46
Encroach Node=108725
       1 2416.54 4719.96
Encroach Node=107532
       1    2008 5263.36
Encroach Node=104348
       1    2700 6339.09
Encroach Node=96265
       1    3500 7740.77
Encroach Node=95077
       1    4800 8615.35
Encroach Node=91978
       1    5450 9244.69
Encroach Node=83613
       115698.1623541.78
Encroach Node=80593
       117663.4524580.11
Encroach Node=76398
       119159.68   25750
Encroach Node=74608
       119738.14   25050
Encroach Node=72672
       118272.61   23650
Encroach Node=71053
       116468.2122022.37
Encroach Node=68028
       116466.1520209.69
Encroach Node=65984
       110676.3313884.37
Encroach Node=64637
       110786.7314232.38
Encroach Node=62238
       110482.6715115.79
Encroach Node=59702
       110099.3213585.21
Encroach Node=56823
       1 9441.2812644.66
Encroach Node=55303
       1 5772.5211047.28
Encroach Node=53117
       1 4866.64 9628.53
Encroach Node=51036
       1 6666.02 9014.57
Encroach Node=48916
       1 6148.76 8065.83
Encroach Node=46568
       1 6818.38 8587.94
Encroach Node=45073
       1 7097.09 8831.57
Encroach Node=44793
       1 7141.11 8968.54
Encroach Node=43746
       1 6661.05 9426.74
Encroach Node=42372
       1 6553.92 9400.68
Encroach Node=39787
       1   12535   15570
Encroach Node=38724
       113168.5115977.76
Encroach Node=37337
       115822.0418835.12
Encroach Node=35159
       112857.7215480.15
Encroach Node=32786
       1 6529.91 9787.39
Encroach Node=30239
       1  6391.5 9367.52
Encroach Node=28041
       1 8541.6810931.68
Encroach Node=26191
       1 8350.6810681.42
Encroach Node=24046
       111686.8814846.15
Encroach Node=19761
       111763.1714722.77
Encroach Node=17358
       111773.9915913.33
Encroach Node=15600
       113375.8816378.11
Encroach Node=13539
       113525.78   18400
Encroach Node=11371
       113271.83   18550
Encroach Node=9505
       115319.42   19500
Encroach Node=7604
       116509.06   19750
Encroach Node=6288
       117048.12   19600
Computation Interval=1MIN
Output Interval=1HOUR
Instantaneous Interval=1HOUR
Mapping Interval=1HOUR
Computation Time Step Use Courant=        0
Computation Time Step Use Time Series=    0
Computation Time Step Count To Double=0
Computation Time Step Max Doubling=0
Computation Time Step Max Halving=0
Computation Time Step Residence Courant=0
Run HTab= 0
Run UNet= 0
Run Sediment= 0
Run PostProcess= 0
Run WQNet= 0
Run RASMapper= 0
UNET Theta= 1
UNET Theta Warmup= 1
UNET ZTol= 0.02
UNET ZSATol= 0.02
UNET MxIter= 20
UNET Max Iter WO Improvement= 0
UNET MaxInSteps= 0
UNET DtIC= 0
UNET DtMin= 0
UNET MaxCRTS= 20
UNET WFStab= 2
UNET SFStab= 1
UNET WFX= 1
UNET SFX= 1
UNET 1D Methodology=Finite Difference
UNET DSS MLevel= 4
UNET Pardiso=0
UNET DZMax Abort= 100
UNET Use Existing IB Tables=-1
UNET Froude Reduction=False
UNET Froude Limit= 0.8
UNET Froude Power= 4
UNET D1 Cores= 0
UNET D2 Coriolis=0
UNET D2 Cores= 0
UNET D2 Theta= 1
UNET D2 Theta Warmup= 1
UNET D2 Z Tol= 0.01
UNET D2 Volume Tol= 0.01
UNET D2 Max Iterations= 20
UNET D2 Equation= 0
UNET D2 RampUpFraction=0.1
UNET D2 TimeSlices= 1
UNET D2 BCVolumeCheck=0
UNET D1D2 MaxIter= 0
UNET D1D2 ZTol=0.01
UNET D1D2 QTol=0.1
UNET D1D2 MinQTol=1
Write IC File= 0
Write IC File at Fixed DateTime=0
Write IC File at Sim End=0
Echo Input=False
Echo Parameters=False
Echo Output=False
Write Detailed= 0
HDF Write Warmup=0
HDF Write Time Slices=0
HDF Flush=0
HDF Face Node Velocities=0
HDF Compression= 1
HDF Chunk Size= 1
HDF Spatial Parts= 1
HDF Use Max Rows=0
HDF Fixed Rows= 1
Calibration Method= 0
Calibration Iterations= 20
Calibration Max Change=0.05
Calibration Tolerance=0.2
Calibration Maximum=1.5
Calibration Minimum=0.5
Calibration Optimization Method= 1
WQ AD Non Conservative
WQ ULTIMATE=-1
WQ Max Comp Step=1HOUR
WQ Output Interval=15MIN
WQ Output Selected Increments= 0
WQ Output face flow=0
WQ Output face velocity=0
WQ Output face area=0
WQ Output face dispersion=0
WQ Output cell volume=0
WQ Output cell surface area=0
WQ Output cell continuity=0
WQ Output cumulative cell continuity=0
WQ Output face conc=0
WQ Output face dconc_dx=0
WQ Output face courant=0
WQ Output face peclet=0
WQ Output face adv mass=0
WQ Output face disp mass=0
WQ Output cell mass=0
WQ Output cell source sink temp=0
WQ Output nsm pathways=0
WQ Output nsm derived pathways=0
WQ Output MaxMinRange=-1
WQ Daily Max Min Mean=-1
WQ Daily Range=0
WQ Daily Time=0
WQ Create Restart=0
WQ Fixed Restart=0
WQ System Summary=0
WQ Write To DSS=0
WQ Use Fixed Temperature=0
Sorting and Armoring Iterations= 10
XS Update Threshold= 0.02
Bed Roughness Predictor= 0
Hydraulics Update Threshold= 0.02
Energy Slope Method= 1
Volume Change Method= 1
Sediment Retention Method= 0
XS Weighting Method= 0
Number of US Weighted Cross Sections= 1
Number of DS Weighted Cross Sections= 1
Upstream XS Weight=0
Main XS Weight=1
Downstream XS Weight=0
Number of DS XS's Weighted with US Boundary= 1
Upstream Boundary Weight= 1
Weight of XSs Associated with US Boundary= 0
Number of US XS's Weighted with DS Boundary= 1
Downstream Boundary Weight= 0.5
Weight of XSs Associated with DS Boundary= 0.5
Percentile Method= 0
Sediment Output Level= 3
Mass or Volume Output= 0
Output Increment Type= 1
Profile and TS Output Increment= 1
XS Output Flag= 0
XS Output Increment= 10
Write Gradation File= 0
Read Gradation Hotstart= 0
Write HDF5 File= 1
Write Binary Output= 1
Write DSS Sediment File= 0
SV Curve= 0
Specific Gage Flag= 0

--- TR_FEMA.p01 (plan) ---

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Plan Title=Trinity_WithLevee
Short Identifier=WithLevee
Geom File=g01
Flow File=f02
Split Flow NTrial= 50
Split Flow Ratio= 0.05
Encroach Param=-1 ,0,0, 0
BEGIN DESCRIPTION:
Geometric data - All hydraulically significant non-accredited levees represented using levee points and IFAs
Flow data - Reduced discharges throughout based on With Levee supplemental model that used lateral structures to represent hydraulically significant non-accredited levees
Boundary condition - Known WS based on With Levee supplemental model
END DESCRIPTION:
DSS File=dss

--- TR_FEMA.p02 (plan) ---

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Plan Title=ScenarioA_Trinity_KaufLID1_HendLID1_NV
Short Identifier=ScenarioA_NV
Geom File=g03
Flow File=f03
Split Flow NTrial= 50
Split Flow Ratio= 0.05
Encroach Param=-1 ,0,0, 0
BEGIN DESCRIPTION:
Geometric data - Kaufman LID1/Henderson LID1 as natural valley and all other hydraulically significant non-accredited levees represented using levee points and IFAs
Flow data - Full discharges through Kaufman LID1/Henderson LID1 with reduced discharges elsewhere based on With Levee supplemental model
Boundary condition - Known WS based on Kaufman LID1/Henderson LID1 supplemental model
END DESCRIPTION:
DSS File=dss

--- TR_FEMA.p03 (plan) ---

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Plan Title=ScenarioB_Trinity_EllisLID2_NV
Short Identifier=ScenarioB_NV
Geom File=g04
Flow File=f05
Split Flow NTrial= 50
Split Flow Ratio= 0.05
Encroach Param=-1 ,0,0, 0
BEGIN DESCRIPTION:
Geometric data - Ellis LID 2 as natural valley and all other hydraulically significant non-accredited levees represented using levee points and IFAs
Flow data - Full discharges through Ellis LID 2 with reduced discharges elsewhere based on With Levee supplemental model
Boundary condition - Known WS based on Ellis LID 2 supplemental model
END DESCRIPTION:
DSS File=dss

--- TR_FEMA.p04 (plan) ---

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Plan Title=ScenarioC_Trinity_KaufMUD1_NV
Short Identifier=ScenarioC_NV
Geom File=g05
Flow File=f06
Split Flow NTrial= 50
Split Flow Ratio= 0.05
Encroach Param=-1 ,0,0, 0
BEGIN DESCRIPTION:
Geometric data - Kaufman MUD 1 as natural valley and all other hydraulically significant non-accredited levees represented using levee points and IFAs
Flow data - Full discharges through Kaufman MUD 1 with reduced discharges elsewhere based on With Levee supplemental model
END DESCRIPTION:
DSS File=dss

--- TR_FEMA.p05 (plan) ---

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Plan Title=ScenarioD_Trinity_Dallas14_Ellis3_NV
Short Identifier=ScenarioD_NV
Geom File=g06
Flow File=f07
Split Flow NTrial= 50
Split Flow Ratio= 0.05
Encroach Param=-1 ,0,0, 0
Optimized Weir=Trinity River   ,1               ,204527
Optimized Weir=Trinity River   ,1               ,148767
Optimized Weir=Trinity River   ,1               ,112555.9
Optimized Weir=Trinity River   ,1               ,83612
Optimized Weir=Trinity River   ,1               ,71044
Optimized Weir=Trinity River   ,1               ,55302
Optimized Weir=Trinity River   ,1               ,51035
BEGIN DESCRIPTION:
Geometric data - Dallas LID14/Ellis LID3 as natural valley and all other hydraulically significant non-accredited levees represented using levee points and IFAs
Flow data - Full discharges through Dallas LID14/Ellis LID3 with reduced discharges elsewhere based on With Levee supplemental model
END DESCRIPTION:
DSS File=dss

--- TR_FEMA.p06 (plan) ---

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Plan Title=ScenarioE_Trinity_BoisDArcLevee_NV
Short Identifier=ScenarioE_NV
Geom File=g07
Flow File=f08
Split Flow NTrial= 50
Split Flow Ratio= 0.05
Encroach Param=-1 ,0,0, 0
Optimized Weir=Trinity River   ,1               ,204527
Optimized Weir=Trinity River   ,1               ,148767
Optimized Weir=Trinity River   ,1               ,112555.9
Optimized Weir=Trinity River   ,1               ,83612
Optimized Weir=Trinity River   ,1               ,71044
Optimized Weir=Trinity River   ,1               ,55302
Optimized Weir=Trinity River   ,1               ,51035
BEGIN DESCRIPTION:
Geometric data - Bois D'Arc Levee as natural valley and all other hydraulically significant non-accredited levees represented using levee points and IFAs
Flow data - Full discharges through Bois D'Arc with reduced discharges elsewhere based on With Levee supplemental model
END DESCRIPTION:
DSS File=dss

--- TR_FEMA.p07 (plan) ---

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Plan Title=ScenarioF_Trinity_DallasLID1_LID2_NV
Short Identifier=ScenarioF_NV
Geom File=g08
Flow File=f09
Split Flow NTrial= 50
Split Flow Ratio= 0.05
Encroach Param=-1 ,0,0, 0
BEGIN DESCRIPTION:
Geometric data - Dallas LID1/Dallas LID2 as natural valley and all other hydraulically significant non-accredited levees represented using levee points and IFAs
Flow data - Full discharges through Dallas LID 1/Dallas LID 2 with reduced discharges elsewhere based on With Levee supplemental model
END DESCRIPTION:
DSS File=dss

--- TR_FEMA.p08 (plan) ---

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Plan Title=Trinity_WithLevee_FW
Short Identifier=WithLevee_FW
Geom File=g01
Flow File=f01
Split Flow NTrial= 50
Split Flow Ratio= 0.05
       111531.9415849.58
       112186.5215042.98
       111895.2413876.77
       111797.0713720.65
       1   1258814525.15
       113923.9216149.17
       113862.0616521.31
       115621.3517812.09
       117978.6520921.35
       118193.7920423.79
       120807.6622930.59
       120792.7722865.83
       119500.4121379.67
       1 17308.419711.52
       113460.0815617.55
       113289.1915534.78
       110296.0913805.69
       113195.6316649.41
       114957.6717013.93
       116867.1919010.01
       1 18246.320585.91
       118473.1420599.72
       115135.9417150.04
       115899.0317892.38
       115913.2117921.79
       116083.7318283.99
       117774.1220414.93
       118057.0420600.43
       117986.2620714.75
DSS File=dss

--- TR_FEMA.p09 (plan) ---

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Plan Title=ScenarioA_KaufLID1_HendLID1_NV_FW
Short Identifier=ScenarioA_FW
Geom File=g03
Flow File=f10
Split Flow NTrial= 50
Split Flow Ratio= 0.05
       1    560011047.28
       1    3950 9628.53
       1    3250 9014.57
       1    2100 8065.83
       1    2000 8587.94
       1    1375 8831.57
       1    1375 8968.54
       1    1000 9426.74
       1     900 9400.68
       1    5900   15570
       1    620015977.76
       1    830018835.12
       1    700015480.15
       1    2600 9787.39
       1    1700 9367.52
       1    220010931.68
       1    180010681.42
       1    550014846.15
       1    520014722.77
       1    490015913.33
       1    450016378.11
       1    4000   18400
       1    3700   18550
       1    4700   19500
       1    5200   19750
       1    5500   19600
DSS File=dss

--- TR_FEMA.p10 (plan) ---

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Plan Title=ScenarioB_EllisLID2_NV_FW
Short Identifier=ScenarioB_FW
Geom File=g04
Flow File=f11
       116468.21   22540
       116466.15   21900
       110676.33   16150
       110786.73   17325
       110482.67   18737
       110099.32   19967
       1 9441.28   20271
       1 5772.52   19335
       1 4866.64   21400
       1 6666.02   20500
       1 6148.76   19000
       1 6818.38   18650
       1 7097.09   18200
       1 7141.11   18200
       1 6661.05   17900
       1 6553.92   17900
       1   12535   24000
       113168.51   24600
       115822.04   27300
       112857.72   24300
       1 6529.91   18700
       1  6391.5   17000
       1 8541.68   18100
       1 8350.68   17850
       111686.88   22300
       111763.17   22100
       111773.99   21200
       113375.88   19600

--- TR_FEMA.p11 (plan) ---

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Plan Title=ScenarioC_KaufMUD1_NV_FW
Short Identifier=ScenarioC_FW
Geom File=g05
Flow File=f12
       1    715023541.78
       1    835024580.11
       1    9900   25750
       1   10300   25050
       1    9300   23650
       1    970022022.37
       1   1170020209.69
       1    700013884.37
       1    730014232.38
       1    760015115.79
       1    740013585.21
       1    740012644.66

--- TR_FEMA.f15 (steady flow) ---

Flow Title=2020 DAlLID1LID2 Reduced Discharges_FW
Program Version=5.06
Number of Profiles= 2
Profile Names=100yr,FW
River Rch & RM=Trinity River,1               ,205777
  120200  120200
River Rch & RM=Trinity River,1               ,200569
  120200  120200
River Rch & RM=Trinity River,1               ,198513
  120200  120200
River Rch & RM=Trinity River,1               ,196991
  120200  120200
River Rch & RM=Trinity River,1               ,195872
  120200  120200
River Rch & RM=Trinity River,1               ,194145
  120200  120200
River Rch & RM=Trinity River,1               ,193094
  120200  120200
River Rch & RM=Trinity River,1               ,191491
  120200  120200
River Rch & RM=Trinity River,1               ,189380
  120200  120200
River Rch & RM=Trinity River,1               ,187750
  120200  120200
River Rch & RM=Trinity River,1               ,186516
  120200  120200
River Rch & RM=Trinity River,1               ,186264
  120200  120200
River Rch & RM=Trinity River,1               ,184503
  120200  120200
River Rch & RM=Trinity River,1               ,181750
  120200  120200
River Rch & RM=Trinity River,1               ,179572
  120200  120200
River Rch & RM=Trinity River,1               ,178698
  120200  120200
River Rch & RM=Trinity River,1               ,176021
  108900  108900
River Rch & RM=Trinity River,1               ,172483
  108900  108900
River Rch & RM=Trinity River,1               ,169025
  108900  108900
River Rch & RM=Trinity River,1               ,167085
  108900  108900
River Rch & RM=Trinity River,1               ,165454
  108900  108900
River Rch & RM=Trinity River,1               ,165204
  108900  108900
River Rch & RM=Trinity River,1               ,164199
  108900  108900
River Rch & RM=Trinity River,1               ,162832
  108900  108900
River Rch & RM=Trinity River,1               ,161707
  108900  108900
River Rch & RM=Trinity River,1               ,159456
  108900  108900
River Rch & RM=Trinity River,1               ,157344
  108900  108900
River Rch & RM=Trinity River,1               ,154267
  109800  109800
River Rch & RM=Trinity River,1               ,151264
  109800  109800
River Rch & RM=Trinity River,1               ,148768
   75646   75646
River Rch & RM=Trinity River,1               ,147333
  101796  101796
River Rch & RM=Trinity River,1               ,145717
  100066  100066
River Rch & RM=Trinity River,1               ,143893
   98353   98353
River Rch & RM=Trinity River,1               ,141890
   96461   96461
River Rch & RM=Trinity River,1               ,139225
   95114   95114
River Rch & RM=Trinity River,1               ,137179
   94221   94221
River Rch & RM=Trinity River,1               ,135104
   92323   92323
River Rch & RM=Trinity River,1               ,133245
   91574   91574
River Rch & RM=Trinity River,1               ,131382
   91110   91110
River Rch & RM=Trinity River,1               ,129561
   89961   89961
River Rch & RM=Trinity River,1               ,127110
   88212   88212
River Rch & RM=Trinity River,1               ,124996
   87518   87518
River Rch & RM=Trinity River,1               ,123554
   86865   86865
River Rch & RM=Trinity River,1               ,122155
   86289   86289
River Rch & RM=Trinity River,1               ,120905
   85471   85471
River Rch & RM=Trinity River,1               ,118211
   85149   85149
River Rch & RM=Trinity River,1               ,116211
   85099   85099
River Rch & RM=Trinity River,1               ,113969
   80343   80343
River Rch & RM=Trinity River,1               ,112556
   79867   79867
River Rch & RM=Trinity River,1               ,110130
   79694   79694
River Rch & RM=Trinity River,1               ,108725
   79650   79650
River Rch & RM=Trinity River,1               ,107532
   79394   79394
River Rch & RM=Trinity River,1               ,104348
   84781   84781
River Rch & RM=Trinity River,1               ,96265
   83325   83325
River Rch & RM=Trinity River,1               ,95077
   82957   82957
River Rch & RM=Trinity River,1               ,91978
   82047   82047
River Rch & RM=Trinity River,1               ,83613
  115869  115869
River Rch & RM=Trinity River,1               ,80593
  118346  118346
River Rch & RM=Trinity River,1               ,76398
  117395  117395
River Rch & RM=Trinity River,1               ,74608
  138421  138421
River Rch & RM=Trinity River,1               ,72672
  137070  137070
River Rch & RM=Trinity River,1               ,71053
  135335  135335
River Rch & RM=Trinity River,1               ,68028
  132522  132522
River Rch & RM=Trinity River,1               ,65984
  129170  129170
River Rch & RM=Trinity River,1               ,64637
  127365  127365
River Rch & RM=Trinity River,1               ,62238
  125051  125051
River Rch & RM=Trinity River,1               ,59702
  120222  120222
River Rch & RM=Trinity River,1               ,56823
  118920  118920
River Rch & RM=Trinity River,1               ,55303
  118888  118888
River Rch & RM=Trinity River,1               ,53117
  131796  131796
River Rch & RM=Trinity River,1               ,51036
  130576  130576
River Rch & RM=Trinity River,1               ,48916
  126168  126168
River Rch & RM=Trinity River,1               ,46568
  123596  123596
River Rch & RM=Trinity River,1               ,45073
  121544  121544
River Rch & RM=Trinity River,1               ,44793
  121544  121544
River Rch & RM=Trinity River,1               ,43746
  120399  120399
River Rch & RM=Trinity River,1               ,42372
  117205  117205
River Rch & RM=Trinity River,1               ,39787
  115868  115868
River Rch & RM=Trinity River,1               ,38724
  113963  113963
River Rch & RM=Trinity River,1               ,37337
  112342  112342
River Rch & RM=Trinity River,1               ,35159
  109477  109477
River Rch & RM=Trinity River,1               ,32786
  109217  109217
River Rch & RM=Trinity River,1               ,30239
  108396  108396
River Rch & RM=Trinity River,1               ,28041
  107960  107960
River Rch & RM=Trinity River,1               ,26191
  106827  106827
River Rch & RM=Trinity River,1               ,24046
  106502  106502
River Rch & RM=Trinity River,1               ,19761
  106502  106502
River Rch & RM=Trinity River,1               ,17358
  105875  105875
River Rch & RM=Trinity River,1               ,15600
  105768  105768
River Rch & RM=Trinity River,1               ,13539
  105742  105742
River Rch & RM=Trinity River,1               ,11371
  133942  133942
River Rch & RM=Trinity River,1               ,9505
  133677  133677
River Rch & RM=Trinity River,1               ,7604
  133585  133585
River Rch & RM=Trinity River,1               ,6288
  133542  133542
Boundary for River Rch & Prof#=Trinity River,1               , 1
Up Type= 0
Dn Type= 1
Dn Known WS=329.3
Boundary for River Rch & Prof#=Trinity River,1               , 2
Up Type= 0
Dn Type= 1
Dn Known WS=329.3
DSS Import GetInterval= 0
DSS Import GetPeak= 0
DSS Import FillOption= 0

--- TR_FEMA.f01 (steady flow) ---

Flow Title=2020 USACE Reduced Trinity Discharges_FW
Program Version=5.06
Number of Profiles= 2
Profile Names=100yr,FW
River Rch & RM=Trinity River,1               ,205777
  120200  120200
River Rch & RM=Trinity River,1               ,200569
  117604  117604
River Rch & RM=Trinity River,1               ,198513
  115435  115435
River Rch & RM=Trinity River,1               ,196991
  113486  113486
River Rch & RM=Trinity River,1               ,195872
  112383  112383
River Rch & RM=Trinity River,1               ,194145
  110743  110743
River Rch & RM=Trinity River,1               ,193094
  110146  110146
River Rch & RM=Trinity River,1               ,191491
  108900  108900
River Rch & RM=Trinity River,1               ,189380
  106968  106968
River Rch & RM=Trinity River,1               ,187750
  104741  104741
River Rch & RM=Trinity River,1               ,186516
  102185  102185
River Rch & RM=Trinity River,1               ,186264
  102185  102185
River Rch & RM=Trinity River,1               ,184503
  100291  100291
River Rch & RM=Trinity River,1               ,181750
   98659   98659
River Rch & RM=Trinity River,1               ,179572
   97745   97745
River Rch & RM=Trinity River,1               ,178698
   97119   97119
River Rch & RM=Trinity River,1               ,176021
   85208   85208
River Rch & RM=Trinity River,1               ,172483
   84264   84264
River Rch & RM=Trinity River,1               ,169025
   83032   83032
River Rch & RM=Trinity River,1               ,167085
   81420   81420
River Rch & RM=Trinity River,1               ,165454
   80056   80056
River Rch & RM=Trinity River,1               ,165204
   80056   80056
River Rch & RM=Trinity River,1               ,164199
   79708   79708
River Rch & RM=Trinity River,1               ,162832
   79382   79382
River Rch & RM=Trinity River,1               ,161707
   78205   78205
River Rch & RM=Trinity River,1               ,159456
   76383   76383
River Rch & RM=Trinity River,1               ,157344
   75613   75613
River Rch & RM=Trinity River,1               ,154267
   75896   75896
River Rch & RM=Trinity River,1               ,151264
   75677   75677
River Rch & RM=Trinity River,1               ,148768
   75646   75646
River Rch & RM=Trinity River,1               ,147333
  101796  101796
River Rch & RM=Trinity River,1               ,145717
  100066  100066
River Rch & RM=Trinity River,1               ,143893
   98353   98353
River Rch & RM=Trinity River,1               ,141890
   96461   96461
River Rch & RM=Trinity River,1               ,139225
   95114   95114
River Rch & RM=Trinity River,1               ,137179
   94221   94221
River Rch & RM=Trinity River,1               ,135104
   92323   92323
River Rch & RM=Trinity River,1               ,133245
   91574   91574
River Rch & RM=Trinity River,1               ,131382
   91110   91110
River Rch & RM=Trinity River,1               ,129561
   89961   89961
River Rch & RM=Trinity River,1               ,127110
   88212   88212
River Rch & RM=Trinity River,1               ,124996
   87518   87518
River Rch & RM=Trinity River,1               ,123554
   86865   86865
River Rch & RM=Trinity River,1               ,122155
   86289   86289
River Rch & RM=Trinity River,1               ,120905
   85471   85471
River Rch & RM=Trinity River,1               ,118211
   85149   85149
River Rch & RM=Trinity River,1               ,116211
   85099   85099
River Rch & RM=Trinity River,1               ,113969
   80343   80343
River Rch & RM=Trinity River,1               ,112556
   79867   79867
River Rch & RM=Trinity River,1               ,110130
   79694   79694
River Rch & RM=Trinity River,1               ,108725
   79650   79650
River Rch & RM=Trinity River,1               ,107532
   79394   79394
River Rch & RM=Trinity River,1               ,104348
   84781   84781
River Rch & RM=Trinity River,1               ,96265
   83325   83325
River Rch & RM=Trinity River,1               ,95077
   82957   82957
River Rch & RM=Trinity River,1               ,91978
   82047   82047
River Rch & RM=Trinity River,1               ,83613
  115869  115869
River Rch & RM=Trinity River,1               ,80593
  118346  118346
River Rch & RM=Trinity River,1               ,76398
  117395  117395
River Rch & RM=Trinity River,1               ,74608
  138421  138421
River Rch & RM=Trinity River,1               ,72672
  137070  137070
River Rch & RM=Trinity River,1               ,71053
  135335  135335
River Rch & RM=Trinity River,1               ,68028
  132522  132522
River Rch & RM=Trinity River,1               ,65984
  129170  129170
River Rch & RM=Trinity River,1               ,64637
  127365  127365
River Rch & RM=Trinity River,1               ,62238
  125051  125051
River Rch & RM=Trinity River,1               ,59702
  120222  120222
River Rch & RM=Trinity River,1               ,56823
  118920  118920
River Rch & RM=Trinity River,1               ,55303
  118888  118888
River Rch & RM=Trinity River,1               ,53117
  131796  131796
River Rch & RM=Trinity River,1               ,51036
  130576  130576
River Rch & RM=Trinity River,1               ,48916
  126168  126168
River Rch & RM=Trinity River,1               ,46568
  123596  123596
River Rch & RM=Trinity River,1               ,45073
  121544  121544
River Rch & RM=Trinity River,1               ,44793
  121544  121544
River Rch & RM=Trinity River,1               ,43746
  120399  120399
River Rch & RM=Trinity River,1               ,42372
  117205  117205
River Rch & RM=Trinity River,1               ,39787
  115868  115868
River Rch & RM=Trinity River,1               ,38724
  113963  113963
River Rch & RM=Trinity River,1               ,37337
  112342  112342
River Rch & RM=Trinity River,1               ,35159
  109477  109477
River Rch & RM=Trinity River,1               ,32786
  109217  109217
River Rch & RM=Trinity River,1               ,30239
  108396  108396
River Rch & RM=Trinity River,1               ,28041
  107960  107960
River Rch & RM=Trinity River,1               ,26191
  106827  106827
River Rch & RM=Trinity River,1               ,24046
  106502  106502
River Rch & RM=Trinity River,1               ,19761
  106502  106502
River Rch & RM=Trinity River,1               ,17358
  105875  105875
River Rch & RM=Trinity River,1               ,15600
  105768  105768
River Rch & RM=Trinity River,1               ,13539
  105742  105742
River Rch & RM=Trinity River,1               ,11371
  133942  133942
River Rch & RM=Trinity River,1               ,9505
  133677  133677
River Rch & RM=Trinity River,1               ,7604
  133585  133585
River Rch & RM=Trinity River,1               ,6288
  133542  133542
Boundary for River Rch & Prof#=Trinity River,1               , 1
Up Type= 0
Dn Type= 1
Dn Known WS=329.3
Boundary for River Rch & Prof#=Trinity River,1               , 2
Up Type= 0
Dn Type= 1
Dn Known WS=329.3
DSS Import GetInterval= 0
DSS Import GetPeak= 0
DSS Import FillOption= 0

--- TR_FEMA.f02 (steady flow) ---

Flow Title=2020 USACE Reduced Trinity Discharges
Program Version=5.06
BEGIN FILE DESCRIPTION:
Reduced discharges throughout based on With Levee supplemental model that used lateral structures to represent hydraulically significant non-accredited levees
END FILE DESCRIPTION:
Number of Profiles= 7
Profile Names=10yr,25yr,50yr,100yr,500yr,1PCT_MINUS,1PCT_PLUS
River Rch & RM=Trinity River,1               ,205777
   50100   75100   95700  120200  185200   87400  193600
River Rch & RM=Trinity River,1               ,200569
   50100   75091   94845  117604  177387   87001  184767
River Rch & RM=Trinity River,1               ,198513
   50100   75059   94005  115435  171504   86543  178140
River Rch & RM=Trinity River,1               ,196991
   50100   74828   93020  113486  167115   85860  173248
River Rch & RM=Trinity River,1               ,195872
   50100   74766   92518  112383  164541   85541  170364
River Rch & RM=Trinity River,1               ,194145
   50100   74649   91729  110743  160793   85020  166172
River Rch & RM=Trinity River,1               ,193094
   50100   74595   91432  110146  159532   84818  164766
River Rch & RM=Trinity River,1               ,191491
   50100   74516   90901  108900  156308   84476  160955
River Rch & RM=Trinity River,1               ,189380
   50100   74324   89988  106968  152250   83859  156278
River Rch & RM=Trinity River,1               ,187750
   50100   74041   88838  104741  148012   83042  151481
River Rch & RM=Trinity River,1               ,186516
   50100   73520   87326  102185  143688   81880  146553
River Rch & RM=Trinity River,1               ,186264
   50100   73520   87326  102185  143688   81880  146553
River Rch & RM=Trinity River,1               ,184503
   50100   73288   86436  100291  138200   81216  140477
River Rch & RM=Trinity River,1               ,181750
   50100   73271   85833   98659  132968   80854  134862
River Rch & RM=Trinity River,1               ,179572
   50100   73264   85552   97745  129718   80687  131451
River Rch & RM=Trinity River,1               ,178698
   50100   73264   85343   97119  127830   80562  129511
River Rch & RM=Trinity River,1               ,176021
   44300   64464   75864   85208  107043   73662  104979
River Rch & RM=Trinity River,1               ,172483
   44300   64464   75506   84264  104285   73418  102211
River Rch & RM=Trinity River,1               ,169025
   44300   64333   74951   83032  100582   72978   98662
River Rch & RM=Trinity River,1               ,167085
   44300   64040   74126   81420   96746   72288   94909
River Rch & RM=Trinity River,1               ,165454
   44300   63853   73493   80056   93413   71803   91647
River Rch & RM=Trinity River,1               ,165204
   44300   63853   73493   80056   93413   71803   91647
River Rch & RM=Trinity River,1               ,164199
   44300   63851   73372   79708   92019   71723   90329
River Rch & RM=Trinity River,1               ,162832
   44300   63848   73304   79382   90383   71680   88788
River Rch & RM=Trinity River,1               ,161707
   44300   63744   72732   78205   87601   71238   86073
River Rch & RM=Trinity River,1               ,159456
   44300   63597   71853   76383   83295   70567   81877
River Rch & RM=Trinity River,1               ,157344
   44300   63560   71536   75613   80665   70328   79284
River Rch & RM=Trinity River,1               ,154267
   44700   64260   72098   75896   79419   70858   78497
River Rch & RM=Trinity River,1               ,151264
   44700   64260   72095   75677   77074   70858   76106
River Rch & RM=Trinity River,1               ,148768
   44700   64260   72094   75646   76784   70858   75808
River Rch & RM=Trinity River,1               ,147333
   44700   66256   84088  101796  139875   79117  142868
River Rch & RM=Trinity River,1               ,145717
   44700   66228   83478  100066  134896   78712  137782
River Rch & RM=Trinity River,1               ,143893
   44700   66210   82907   98353  130099   78365  132907
River Rch & RM=Trinity River,1               ,141890
   44700   66207   82210   96461  125161   77933  127939
River Rch & RM=Trinity River,1               ,139225
   44700   66193   81673   95114  121844   77576  124666
River Rch & RM=Trinity River,1               ,137179
   44700   66182   81303   94221  119519   77320  122422
River Rch & RM=Trinity River,1               ,135104
   44700   66070   80442   92323  114967   76661  118012
River Rch & RM=Trinity River,1               ,133245
   44700   66070   80212   91574  112562   76521  115753
River Rch & RM=Trinity River,1               ,131382
   44700   66070   80113   91110  110670   76464  114010
River Rch & RM=Trinity River,1               ,129561
   44700   66049   79722   89961  107630   76194  111103
River Rch & RM=Trinity River,1               ,127110
   44700   65815   78807   88212  104089   75429  107679
River Rch & RM=Trinity River,1               ,124996
   44700   65743   78512   87518  102003   75176  105712
River Rch & RM=Trinity River,1               ,123554
   44700   65742   78271   86865  100204   74991  104042
River Rch & RM=Trinity River,1               ,122155
   44700   65729   78023   86289   98891   74783  102800
River Rch & RM=Trinity River,1               ,120905
   44700   65695   77673   85471   97034   74485  101039
River Rch & RM=Trinity River,1               ,118211
   44700   65695   77587   85149   95921   74416  100001
River Rch & RM=Trinity River,1               ,116211
   44700   65695   77575   85099   95457   74405   99637
River Rch & RM=Trinity River,1               ,113969
   40000   61295   71398   80343   87595   72241   88631
River Rch & RM=Trinity River,1               ,112556
   40000   61291   71281   79867   85924   72142   87038
River Rch & RM=Trinity River,1               ,110130
   40000   61291   71269   79694   85126   72132   86276
River Rch & RM=Trinity River,1               ,108725
   40000   61291   71269   79650   84751   72132   85924
River Rch & RM=Trinity River,1               ,107532
   40000   61291   71262   79394   83402   72131   84529
River Rch & RM=Trinity River,1               ,104348
   40000   62008   73422   84781  106737   73589  109056
River Rch & RM=Trinity River,1               ,96265
   40000   62005   73273   83325   99225   73526  101078
River Rch & RM=Trinity River,1               ,95077
   40000   62005   73246   82957   97670   73518   99415
River Rch & RM=Trinity River,1               ,91978
   40000   62000   73037   82047   94619   73393   96168
River Rch & RM=Trinity River,1               ,83613
   56100   86267  102499  115869  147207   98335  150100
River Rch & RM=Trinity River,1               ,80593
   56100   86297  103199  118346  156321   98860  159388
River Rch & RM=Trinity River,1               ,76398
   56100   86297  102909  117395  153572   98669  156563
River Rch & RM=Trinity River,1               ,74608
   56100   86900  110479  138421  209309  104114  212555
River Rch & RM=Trinity River,1               ,72672
   56100   86896  109963  137070  205824  103731  208981
River Rch & RM=Trinity River,1               ,71053
   56100   86861  109210  135335  201676  103136  204734
River Rch & RM=Trinity River,1               ,68028
   56100   86838  108124  132522  192141  102287  194934
River Rch & RM=Trinity River,1               ,65984
   56100   86836  107011  129170  182626  101459  185223
River Rch & RM=Trinity River,1               ,64637
   56100   86834  106583  127365  176781  101167  179271
River Rch & RM=Trinity River,1               ,62238
   56100   86831  105966  125051  169878  100728  172248
River Rch & RM=Trinity River,1               ,59702
   56100   86800  104338  120222  156737   99453  158935
River Rch & RM=Trinity River,1               ,56823
   56100   86800  103899  118920  152495   99098  154591
River Rch & RM=Trinity River,1               ,55303
   56100   86800  103899  118888  151146   99098  153198
River Rch & RM=Trinity River,1               ,53117
   56100   86875  109244  131796  181011  103218  183863
River Rch & RM=Trinity River,1               ,51036
   56100   86875  109005  130576  176441  103046  179203
River Rch & RM=Trinity River,1               ,48916
   51600   78575  102701  126168  167459  100774  168767
River Rch & RM=Trinity River,1               ,46568
   51600   78575  102301  123596  159545  100474  160751
River Rch & RM=Trinity River,1               ,45073
   51600   78575  101772  121544  154452  100036  155579
River Rch & RM=Trinity River,1               ,44793
   51600   78575  101772  121544  154452  100036  155579
River Rch & RM=Trinity River,1               ,43746
   51600   78575  101397  120399  151548   99708  152598
River Rch & RM=Trinity River,1               ,42372
   51600   78403   99736  117205  145757   98179  146712
River Rch & RM=Trinity River,1               ,39787
   51600   78400   99218  115868  142484   97711  143359
River Rch & RM=Trinity River,1               ,38724
   51600   78375   98359  113963  138763   96928  139570
River Rch & RM=Trinity River,1               ,37337
   51600   78266   97508  112342  135723   96140  136463
River Rch & RM=Trinity River,1               ,35159
   51600   77976   96109  109477  130089   94854  130684
River Rch & RM=Trinity River,1               ,32786
   51600   77976   96085  109217  128917   94838  129436
River Rch & RM=Trinity River,1               ,30239
   51600   77976   95951  108396  126459   94736  126840
River Rch & RM=Trinity River,1               ,28041
   51600   77976   95899  107960  124932   94696  125230
River Rch & RM=Trinity River,1               ,26191
   51600   77975   95621  106827  121908   94467  122064
River Rch & RM=Trinity River,1               ,24046
   51600   77975   95591  106502  120583   94451  120641
River Rch & RM=Trinity River,1               ,19761
   51600   77975   95591  106502  120357   94451  120374
River Rch & RM=Trinity River,1               ,17358
   51600   77975   95488  105875  118183   94379  118115
River Rch & RM=Trinity River,1               ,15600
   51600   77975   95488  105768  116821   94379  116665
River Rch & RM=Trinity River,1               ,13539
   51600   77975   95488  105742  116296   94379  116118
River Rch & RM=Trinity River,1               ,11371
   51600   78600  104501  133942  196620  102015  198170
River Rch & RM=Trinity River,1               ,9505
   51600   78600  104500  133677  195527  102015  197064
River Rch & RM=Trinity River,1               ,7604
   51600   78600  104500  133585  194701  102015  196225
River Rch & RM=Trinity River,1               ,6288
   51600   78600  104500  133542  194157  102015  195673
Boundary for River Rch & Prof#=Trinity River,1               , 1
Up Type= 0
Dn Type= 1
Dn Known WS=322.4
Boundary for River Rch & Prof#=Trinity River,1               , 2
Up Type= 0
Dn Type= 1
Dn Known WS=325.55
Boundary for River Rch & Prof#=Trinity River,1               , 3
Up Type= 0
Dn Type= 1
Dn Known WS=327.49
Boundary for River Rch & Prof#=Trinity River,1               , 4
Up Type= 0
Dn Type= 1
Dn Known WS=329.3
Boundary for River Rch & Prof#=Trinity River,1               , 5
Up Type= 0
Dn Type= 1
Dn Known WS=332.4
Boundary for River Rch & Prof#=Trinity River,1               , 6
Up Type= 0
Dn Type= 1
Dn Known WS=327.32
Boundary for River Rch & Prof#=Trinity River,1               , 7
Up Type= 0
Dn Type= 1
Dn Known WS=332.47
DSS Import GetInterval= 0
DSS Import GetPeak= 0
DSS Import FillOption= 0
