HEC-RAS study TR_FEMA.prj: Trinity_River_FEMA

--- TR_FEMA.f03 (steady flow) ---

Flow Title=2020 KaufHendLID1 Reduced Discharges
Program Version=5.06
BEGIN FILE DESCRIPTION:
Full discharges through Kaufman LID1/Henderson LID1 with reduced discharges elsewhere based on With Levee supplemental model that used lateral structures to represent levees
Boundary condition - Known WS based on Kaufman LID1/Henderson LID1 supplemental model
END FILE DESCRIPTION:
Number of Profiles= 7
Profile Names=10yr,25yr,50yr,100yr,500yr,1PCT_MINUS,1PCT_PLUS
River Rch & RM=Trinity River,1               ,205777
   50100   75100   95700  120200  185200   87400  193600
River Rch & RM=Trinity River,1               ,200569
   50100   75091   94845  117604  177387   87001  184767
River Rch & RM=Trinity River,1               ,198513
   50100   75059   94005  115435  171504   86543  178140
River Rch & RM=Trinity River,1               ,196991
   50100   74828   93020  113486  167115   85860  173248
River Rch & RM=Trinity River,1               ,195872
   50100   74766   92518  112383  164541   85541  170364
River Rch & RM=Trinity River,1               ,194145
   50100   74649   91729  110743  160793   85020  166172
River Rch & RM=Trinity River,1               ,193094
   50100   74595   91432  110146  159532   84818  164766
River Rch & RM=Trinity River,1               ,191491
   50100   74516   90901  108900  156308   84476  160955
River Rch & RM=Trinity River,1               ,189380
   50100   74324   89988  106968  152250   83859  156278
River Rch & RM=Trinity River,1               ,187750
   50100   74041   88838  104741  148012   83042  151481
River Rch & RM=Trinity River,1               ,186516
   50100   73520   87326  102185  143688   81880  146553
River Rch & RM=Trinity River,1               ,186264
   50100   73520   87326  102185  143688   81880  146553
River Rch & RM=Trinity River,1               ,184503
   50100   73288   86436  100291  138200   81216  140477
River Rch & RM=Trinity River,1               ,181750
   50100   73271   85833   98659  132968   80854  134862
River Rch & RM=Trinity River,1               ,179572
   50100   73264   85552   97745  129718   80687  131451
River Rch & RM=Trinity River,1               ,178698
   50100   73264   85343   97119  127830   80562  129511
River Rch & RM=Trinity River,1               ,176021
   44300   64464   75864   85208  107043   73662  104979
River Rch & RM=Trinity River,1               ,172483
   44300   64464   75506   84264  104285   73418  102211
River Rch & RM=Trinity River,1               ,169025
   44300   64333   74951   83032  100582   72978   98662
River Rch & RM=Trinity River,1               ,167085
   44300   64040   74126   81420   96746   72288   94909
River Rch & RM=Trinity River,1               ,165454
   44300   63853   73493   80056   93413   71803   91647
River Rch & RM=Trinity River,1               ,165204
   44300   63853   73493   80056   93413   71803   91647
River Rch & RM=Trinity River,1               ,164199
   44300   63851   73372   79708   92019   71723   90329
River Rch & RM=Trinity River,1               ,162832
   44300   63848   73304   79382   90383   71680   88788
River Rch & RM=Trinity River,1               ,161707
   44300   63744   72732   78205   87601   71238   86073
River Rch & RM=Trinity River,1               ,159456
   44300   63597   71853   76383   83295   70567   81877
River Rch & RM=Trinity River,1               ,157344
   44300   63560   71536   75613   80665   70328   79284
River Rch & RM=Trinity River,1               ,154267
   44700   64260   72098   75896   79419   70858   78497
River Rch & RM=Trinity River,1               ,151264
   44700   64260   72095   75677   77074   70858   76106
River Rch & RM=Trinity River,1               ,148768
   44700   64260   72094   75646   76784   70858   75808
River Rch & RM=Trinity River,1               ,147333
   44700   66256   84088  101796  139875   79117  142868
River Rch & RM=Trinity River,1               ,145717
   44700   66228   83478  100066  134896   78712  137782
River Rch & RM=Trinity River,1               ,143893
   44700   66210   82907   98353  130099   78365  132907
River Rch & RM=Trinity River,1               ,141890
   44700   66207   82210   96461  125161   77933  127939
River Rch & RM=Trinity River,1               ,139225
   44700   66193   81673   95114  121844   77576  124666
River Rch & RM=Trinity River,1               ,137179
   44700   66182   81303   94221  119519   77320  122422
River Rch & RM=Trinity River,1               ,135104
   44700   66070   80442   92323  114967   76661  118012
River Rch & RM=Trinity River,1               ,133245
   44700   66070   80212   91574  112562   76521  115753
River Rch & RM=Trinity River,1               ,131382
   44700   66070   80113   91110  110670   76464  114010
River Rch & RM=Trinity River,1               ,129561
   44700   66049   79722   89961  107630   76194  111103
River Rch & RM=Trinity River,1               ,127110
   44700   65815   78807   88212  104089   75429  107679
River Rch & RM=Trinity River,1               ,124996
   44700   65743   78512   87518  102003   75176  105712
River Rch & RM=Trinity River,1               ,123554
   44700   65742   78271   86865  100204   74991  104042
River Rch & RM=Trinity River,1               ,122155
   44700   65729   78023   86289   98891   74783  102800
River Rch & RM=Trinity River,1               ,120905
   44700   65695   77673   85471   97034   74485  101039
River Rch & RM=Trinity River,1               ,118211
   44700   65695   77587   85149   95921   74416  100001
River Rch & RM=Trinity River,1               ,116211
   44700   65695   77575   85099   95457   74405   99637
River Rch & RM=Trinity River,1               ,113969
   40000   61295   71398   80343   87595   72241   88631
River Rch & RM=Trinity River,1               ,112556
   40000   61291   71281   79867   85924   72142   87038
River Rch & RM=Trinity River,1               ,110130
   40000   61291   71269   79694   85126   72132   86276
River Rch & RM=Trinity River,1               ,108725
   40000   61291   71269   79650   84751   72132   85924
River Rch & RM=Trinity River,1               ,107532
   40000   61291   71262   79394   83402   72131   84529
River Rch & RM=Trinity River,1               ,104348
   40000   62008   73422   84781  106737   73589  109056
River Rch & RM=Trinity River,1               ,96265
   40000   62005   73273   83325   99225   73526  101078
River Rch & RM=Trinity River,1               ,95077
   40000   62005   73246   82957   97670   73518   99415
River Rch & RM=Trinity River,1               ,91978
   40000   62000   73037   82047   94619   73393   96168
River Rch & RM=Trinity River,1               ,83613
   56100   86267  102499  115869  147207   98335  150100
River Rch & RM=Trinity River,1               ,80593
   56100   86297  103199  118346  156321   98860  159388
River Rch & RM=Trinity River,1               ,76398
   56100   86297  102909  117395  153572   98669  156563
River Rch & RM=Trinity River,1               ,74608
   56100   86900  110479  138421  209309  104114  212555
River Rch & RM=Trinity River,1               ,72672
   56100   86896  109963  137070  205824  103731  208981
River Rch & RM=Trinity River,1               ,71053
   56100   86861  109210  135335  201676  103136  204734
River Rch & RM=Trinity River,1               ,68028
   56100   86838  108124  132522  192141  102287  194934
River Rch & RM=Trinity River,1               ,65984
   56100   86836  107011  129170  182626  101459  185223
River Rch & RM=Trinity River,1               ,64637
   56100   86834  106583  127365  176781  101167  179271
River Rch & RM=Trinity River,1               ,62238
   56100   86831  105966  125051  169878  100728  172248
River Rch & RM=Trinity River,1               ,59702
   56100   86800  104338  120222  156737   99453  158935
River Rch & RM=Trinity River,1               ,56823
   56100   86800  103899  118920  152495   99098  154591
River Rch & RM=Trinity River,1               ,55303
   56100   86900  111100  141000  217800  104500  221300
River Rch & RM=Trinity River,1               ,53117
   56100   86900  111100  141000  217800  104500  221300
River Rch & RM=Trinity River,1               ,51036
   56100   86900  111100  141000  217800  104500  221300
River Rch & RM=Trinity River,1               ,48916
   51600   78600  104900  137400  212400  102300  214500
River Rch & RM=Trinity River,1               ,46568
   51600   78600  104900  137400  212400  102300  214500
River Rch & RM=Trinity River,1               ,45073
   51600   78600  104900  137400  212400  102300  214500
River Rch & RM=Trinity River,1               ,44793
   51600   78600  104900  137400  212400  102300  214500
River Rch & RM=Trinity River,1               ,43746
   51600   78600  104900  137400  212400  102300  214500
River Rch & RM=Trinity River,1               ,42372
   51600   78600  104900  137400  212400  102300  214500
River Rch & RM=Trinity River,1               ,39787
   51600   78600  104900  137400  212400  102300  214500
River Rch & RM=Trinity River,1               ,38724
   51600   78600  104900  137400  212400  102300  214500
River Rch & RM=Trinity River,1               ,37337
   51600   78600  104900  137400  212400  102300  214500
River Rch & RM=Trinity River,1               ,35159
   51600   78600  104900  137400  212400  102300  214500
River Rch & RM=Trinity River,1               ,32786
   51600   78600  104900  137400  212400  102300  214500
River Rch & RM=Trinity River,1               ,30239
   51600   78600  104900  137400  212400  102300  214500
River Rch & RM=Trinity River,1               ,28041
   51600   78600  104900  137400  212400  102300  214500
River Rch & RM=Trinity River,1               ,26191
   51600   78600  104900  137400  212400  102300  214500
River Rch & RM=Trinity River,1               ,24046
   51600   78600  104900  137400  212400  102300  214500
River Rch & RM=Trinity River,1               ,19761
   51600   78600  104900  137400  212400  102300  214500
River Rch & RM=Trinity River,1               ,17358
   51600   78600  104900  137400  212400  102300  214500
River Rch & RM=Trinity River,1               ,15600
   51600   78600  104900  137400  212400  102300  214500
River Rch & RM=Trinity River,1               ,13539
   51600   78600  104900  137400  212400  102300  214500
River Rch & RM=Trinity River,1               ,11371
   51600   78600  104900  137400  212400  102300  214500
River Rch & RM=Trinity River,1               ,9505
   51600   78600  104900  137400  212400  102300  214500
River Rch & RM=Trinity River,1               ,7604
   51600   78600  104900  137400  212400  102300  214500
River Rch & RM=Trinity River,1               ,6288
   51600   78600  104900  137400  212400  102300  214500
Boundary for River Rch & Prof#=Trinity River,1               , 1
Up Type= 0
Dn Type= 1
Dn Known WS=316.49
Boundary for River Rch & Prof#=Trinity River,1               , 2
Up Type= 0
Dn Type= 1
Dn Known WS=318.21
Boundary for River Rch & Prof#=Trinity River,1               , 3
Up Type= 0
Dn Type= 1
Dn Known WS=319.63
Boundary for River Rch & Prof#=Trinity River,1               , 4
Up Type= 0
Dn Type= 1
Dn Known WS=321.15
Boundary for River Rch & Prof#=Trinity River,1               , 5
Up Type= 0
Dn Type= 1
Dn Known WS=324.13
Boundary for River Rch & Prof#=Trinity River,1               , 6
Up Type= 0
Dn Type= 1
Dn Known WS=319.5
Boundary for River Rch & Prof#=Trinity River,1               , 7
Up Type= 0
Dn Type= 1
Dn Known WS=324.2
DSS Import GetInterval= 0
DSS Import GetPeak= 0
DSS Import FillOption= 0

--- TR_FEMA.f04 (steady flow) ---

Flow Title=2020 USACE Trinity Discharges
Program Version=5.06
Number of Profiles= 7
Profile Names=10yr,25yr,50yr,100yr,500yr,1PCT_MINUS,1PCT_PLUS
River Rch & RM=Trinity River,1               ,205777
   50100   75100   95700  120200  185200   87400  193600
River Rch & RM=Trinity River,1               ,176021
   44300   66300   86400  108900  166400   80600  171100
River Rch & RM=Trinity River,1               ,154267
   44700   67000   87100  109800  167700   81200  172800
River Rch & RM=Trinity River,1               ,113969
   40000   62600   81000  105400  160900   79100  162800
River Rch & RM=Trinity River,1               ,83613
   56100   86900  111100  141000  217800  104500  221300
River Rch & RM=Trinity River,1               ,48916
   51600   78600  104900  137400  212400  102300  214500
Boundary for River Rch & Prof#=Trinity River,1               , 1
Up Type= 0
Dn Type= 1
Dn Known WS=322.47
Boundary for River Rch & Prof#=Trinity River,1               , 2
Up Type= 0
Dn Type= 1
Dn Known WS=325.59
Boundary for River Rch & Prof#=Trinity River,1               , 3
Up Type= 0
Dn Type= 1
Dn Known WS=327.52
Boundary for River Rch & Prof#=Trinity River,1               , 4
Up Type= 0
Dn Type= 1
Dn Known WS=329.32
Boundary for River Rch & Prof#=Trinity River,1               , 5
Up Type= 0
Dn Type= 1
Dn Known WS=332.41
Boundary for River Rch & Prof#=Trinity River,1               , 6
Up Type= 0
Dn Type= 1
Dn Known WS=327.35
Boundary for River Rch & Prof#=Trinity River,1               , 7
Up Type= 0
Dn Type= 1
Dn Known WS=332.48
DSS Import GetInterval= 0
DSS Import GetPeak= 0
DSS Import FillOption= 0

--- TR_FEMA.f05 (steady flow) ---

Flow Title=2020 EllisLID2 Reduced Discharges
Program Version=5.06
BEGIN FILE DESCRIPTION:
Full discharges through Ellis LID2 with reduced discharges elsewhere based on With Levee supplemental model that used lateral structures to represent hydraulically significant non-accredited levees
Boundary condition - Known WS based on Ellis LID 2 supplemental model
END FILE DESCRIPTION:
Number of Profiles= 7
Profile Names=10yr,25yr,50yr,100yr,500yr,1PCT_MINUS,1PCT_PLUS
River Rch & RM=Trinity River,1               ,205777
   50100   75100   95700  120200  185200   87400  193600
River Rch & RM=Trinity River,1               ,200569
   50100   75091   94845  117604  177387   87001  184767
River Rch & RM=Trinity River,1               ,198513
   50100   75059   94005  115435  171504   86543  178140
River Rch & RM=Trinity River,1               ,196991
   50100   74828   93020  113486  167115   85860  173248
River Rch & RM=Trinity River,1               ,195872
   50100   74766   92518  112383  164541   85541  170364
River Rch & RM=Trinity River,1               ,194145
   50100   74649   91729  110743  160793   85020  166172
River Rch & RM=Trinity River,1               ,193094
   50100   74595   91432  110146  159532   84818  164766
River Rch & RM=Trinity River,1               ,191491
   50100   74516   90901  108900  156308   84476  160955
River Rch & RM=Trinity River,1               ,189380
   50100   74324   89988  106968  152250   83859  156278
River Rch & RM=Trinity River,1               ,187750
   50100   74041   88838  104741  148012   83042  151481
River Rch & RM=Trinity River,1               ,186516
   50100   73520   87326  102185  143688   81880  146553
River Rch & RM=Trinity River,1               ,186264
   50100   73520   87326  102185  143688   81880  146553
River Rch & RM=Trinity River,1               ,184503
   50100   73288   86436  100291  138200   81216  140477
River Rch & RM=Trinity River,1               ,181750
   50100   73271   85833   98659  132968   80854  134862
River Rch & RM=Trinity River,1               ,179572
   50100   73264   85552   97745  129718   80687  131451
River Rch & RM=Trinity River,1               ,178698
   50100   73264   85343   97119  127830   80562  129511
River Rch & RM=Trinity River,1               ,176021
   44300   64464   75864   85208  107043   73662  104979
River Rch & RM=Trinity River,1               ,172483
   44300   64464   75506   84264  104285   73418  102211
River Rch & RM=Trinity River,1               ,169025
   44300   64333   74951   83032  100582   72978   98662
River Rch & RM=Trinity River,1               ,167085
   44300   64040   74126   81420   96746   72288   94909
River Rch & RM=Trinity River,1               ,165454
   44300   63853   73493   80056   93413   71803   91647
River Rch & RM=Trinity River,1               ,165204
   44300   63853   73493   80056   93413   71803   91647
River Rch & RM=Trinity River,1               ,164199
   44300   63851   73372   79708   92019   71723   90329
River Rch & RM=Trinity River,1               ,162832
   44300   63848   73304   79382   90383   71680   88788
River Rch & RM=Trinity River,1               ,161707
   44300   63744   72732   78205   87601   71238   86073
River Rch & RM=Trinity River,1               ,159456
   44300   63597   71853   76383   83295   70567   81877
River Rch & RM=Trinity River,1               ,157344
   44300   63560   71536   75613   80665   70328   79284
River Rch & RM=Trinity River,1               ,154267
   44700   64260   72098   75896   79419   70858   78497
River Rch & RM=Trinity River,1               ,151264
   44700   64260   72095   75677   77074   70858   76106
River Rch & RM=Trinity River,1               ,148768
   44700   64260   72094   75646   76784   70858   75808
River Rch & RM=Trinity River,1               ,147333
   44700   66256   84088  101796  139875   79117  142868
River Rch & RM=Trinity River,1               ,145717
   44700   66228   83478  100066  134896   78712  137782
River Rch & RM=Trinity River,1               ,143893
   44700   66210   82907   98353  130099   78365  132907
River Rch & RM=Trinity River,1               ,141890
   44700   66207   82210   96461  125161   77933  127939
River Rch & RM=Trinity River,1               ,139225
   44700   66193   81673   95114  121844   77576  124666
River Rch & RM=Trinity River,1               ,137179
   44700   66182   81303   94221  119519   77320  122422
River Rch & RM=Trinity River,1               ,135104
   44700   66070   80442   92323  114967   76661  118012
River Rch & RM=Trinity River,1               ,133245
   44700   66070   80212   91574  112562   76521  115753
River Rch & RM=Trinity River,1               ,131382
   44700   66070   80113   91110  110670   76464  114010
River Rch & RM=Trinity River,1               ,129561
   44700   66049   79722   89961  107630   76194  111103
River Rch & RM=Trinity River,1               ,127110
   44700   65815   78807   88212  104089   75429  107679
River Rch & RM=Trinity River,1               ,124996
   44700   65743   78512   87518  102003   75176  105712
River Rch & RM=Trinity River,1               ,123554
   44700   65742   78271   86865  100204   74991  104042
River Rch & RM=Trinity River,1               ,122155
   44700   65729   78023   86289   98891   74783  102800
River Rch & RM=Trinity River,1               ,120905
   44700   65695   77673   85471   97034   74485  101039
River Rch & RM=Trinity River,1               ,118211
   44700   65695   77587   85149   95921   74416  100001
River Rch & RM=Trinity River,1               ,116211
   44700   65695   77575   85099   95457   74405   99637
River Rch & RM=Trinity River,1               ,113969
   40000   61295   71398   80343   87595   72241   88631
River Rch & RM=Trinity River,1               ,112556
   40000   61291   71281   79867   85924   72142   87038
River Rch & RM=Trinity River,1               ,110130
   40000   61291   71269   79694   85126   72132   86276
River Rch & RM=Trinity River,1               ,108725
   40000   61291   71269   79650   84751   72132   85924
River Rch & RM=Trinity River,1               ,107532
   40000   61291   71262   79394   83402   72131   84529
River Rch & RM=Trinity River,1               ,104348
   40000   62008   73422   84781  106737   73589  109056
River Rch & RM=Trinity River,1               ,96265
   40000   62005   73273   83325   99225   73526  101078
River Rch & RM=Trinity River,1               ,95077
   40000   62005   73246   82957   97670   73518   99415
River Rch & RM=Trinity River,1               ,91978
   40000   62000   73037   82047   94619   73393   96168
River Rch & RM=Trinity River,1               ,83613
   56100   86267  102499  115869  147207   98335  150100
River Rch & RM=Trinity River,1               ,80593
   56100   86297  103199  118346  156321   98860  159388
River Rch & RM=Trinity River,1               ,76398
   56100   86297  102909  117395  153572   98669  156563
River Rch & RM=Trinity River,1               ,74608
   56100   86900  110479  138421  209309  104114  212555
River Rch & RM=Trinity River,1               ,72672
   56100   86896  109963  137070  205824  103731  208981
River Rch & RM=Trinity River,1               ,71053
   56100   86900  111100  141000  217800  104500  221300
River Rch & RM=Trinity River,1               ,68028
   56100   86900  111100  141000  217800  104500  221300
River Rch & RM=Trinity River,1               ,65984
   56100   86900  111100  141000  217800  104500  221300
River Rch & RM=Trinity River,1               ,64637
   56100   86900  111100  141000  217800  104500  221300
River Rch & RM=Trinity River,1               ,62238
   56100   86900  111100  141000  217800  104500  221300
River Rch & RM=Trinity River,1               ,59702
   56100   86900  111100  141000  217800  104500  221300
River Rch & RM=Trinity River,1               ,56823
   56100   86900  111100  141000  217800  104500  221300
River Rch & RM=Trinity River,1               ,55303
   56100   86900  111100  141000  217800  104500  221300
River Rch & RM=Trinity River,1               ,53117
   56100   86900  111100  141000  217800  104500  221300
River Rch & RM=Trinity River,1               ,51036
   56100   86900  111100  141000  217800  104500  221300
River Rch & RM=Trinity River,1               ,48916
   51600   78600  104900  137400  212400  102300  214500
River Rch & RM=Trinity River,1               ,46568
   51600   78600  104900  137400  212400  102300  214500
River Rch & RM=Trinity River,1               ,45073
   51600   78600  104900  137400  212400  102300  214500
River Rch & RM=Trinity River,1               ,44793
   51600   78600  104900  137400  212400  102300  214500
River Rch & RM=Trinity River,1               ,43746
   51600   78600  104900  137400  212400  102300  214500
River Rch & RM=Trinity River,1               ,42372
   51600   78600  104900  137400  212400  102300  214500
River Rch & RM=Trinity River,1               ,39787
   51600   78600  104900  137400  212400  102300  214500
River Rch & RM=Trinity River,1               ,38724
   51600   78600  104900  137400  212400  102300  214500
River Rch & RM=Trinity River,1               ,37337
   51600   78600  104900  137400  212400  102300  214500
River Rch & RM=Trinity River,1               ,35159
   51600   78600  104900  137400  212400  102300  214500
River Rch & RM=Trinity River,1               ,32786
   51600   78600  104900  137400  212400  102300  214500
River Rch & RM=Trinity River,1               ,30239
   51600   78600  104900  137400  212400  102300  214500
River Rch & RM=Trinity River,1               ,28041
   51600   78600  104900  137400  212400  102300  214500
River Rch & RM=Trinity River,1               ,26191
   51600   78600  104900  137400  212400  102300  214500
River Rch & RM=Trinity River,1               ,24046
   51600   78600  104900  137400  212400  102300  214500
River Rch & RM=Trinity River,1               ,19761
   51600   78600  104900  137400  212400  102300  214500
River Rch & RM=Trinity River,1               ,17358
   51600   78600  104900  137400  212400  102300  214500
River Rch & RM=Trinity River,1               ,15600
   51600   78600  104900  137400  212400  102300  214500
River Rch & RM=Trinity River,1               ,13539
   51600   77975   95488  105742  116296   94379  116118
River Rch & RM=Trinity River,1               ,11371
   51600   78600  104501  133942  196620  102015  198170
River Rch & RM=Trinity River,1               ,9505
   51600   78600  104500  133677  195527  102015  197064
River Rch & RM=Trinity River,1               ,7604
   51600   78600  104500  133585  194701  102015  196225
River Rch & RM=Trinity River,1               ,6288
   51600   78600  104500  133542  194157  102015  195673
Boundary for River Rch & Prof#=Trinity River,1               , 1
Up Type= 0
Dn Type= 1
Dn Known WS=322.4
Boundary for River Rch & Prof#=Trinity River,1               , 2
Up Type= 0
Dn Type= 1
Dn Known WS=325.55
Boundary for River Rch & Prof#=Trinity River,1               , 3
Up Type= 0
Dn Type= 1
Dn Known WS=327.49
Boundary for River Rch & Prof#=Trinity River,1               , 4
Up Type= 0
Dn Type= 1
Dn Known WS=329.3
Boundary for River Rch & Prof#=Trinity River,1               , 5
Up Type= 0
Dn Type= 1
Dn Known WS=332.4
Boundary for River Rch & Prof#=Trinity River,1               , 6
Up Type= 0
Dn Type= 1
Dn Known WS=327.32
Boundary for River Rch & Prof#=Trinity River,1               , 7
Up Type= 0
Dn Type= 1
Dn Known WS=332.47
DSS Import GetInterval= 0
DSS Import GetPeak= 0
DSS Import FillOption= 0

--- TR_FEMA.f06 (steady flow) ---

Flow Title=2020 KaufMUD1 Reduced Discharges
Program Version=5.06
BEGIN FILE DESCRIPTION:
Full discharges through Kaufman MUD 1with reduced discharges elsewhere based on With Levee supplemental model that used lateral structures to represent levees.
Boundary condition - Known WS based on With Levee supplemental model
END FILE DESCRIPTION:
Number of Profiles= 7
Profile Names=10yr,25yr,50yr,100yr,500yr,1PCT_MINUS,1PCT_PLUS
River Rch & RM=Trinity River,1               ,205777
   50100   75100   95700  120200  185200   87400  193600
River Rch & RM=Trinity River,1               ,200569
   50100   75091   94845  117604  177387   87001  184767
River Rch & RM=Trinity River,1               ,198513
   50100   75059   94005  115435  171504   86543  178140
River Rch & RM=Trinity River,1               ,196991
   50100   74828   93020  113486  167115   85860  173248
River Rch & RM=Trinity River,1               ,195872
   50100   74766   92518  112383  164541   85541  170364
River Rch & RM=Trinity River,1               ,194145
   50100   74649   91729  110743  160793   85020  166172
River Rch & RM=Trinity River,1               ,193094
   50100   74595   91432  110146  159532   84818  164766
River Rch & RM=Trinity River,1               ,191491
   50100   74516   90901  108900  156308   84476  160955
River Rch & RM=Trinity River,1               ,189380
   50100   74324   89988  106968  152250   83859  156278
River Rch & RM=Trinity River,1               ,187750
   50100   74041   88838  104741  148012   83042  151481
River Rch & RM=Trinity River,1               ,186516
   50100   73520   87326  102185  143688   81880  146553
River Rch & RM=Trinity River,1               ,186264
   50100   73520   87326  102185  143688   81880  146553
River Rch & RM=Trinity River,1               ,184503
   50100   73288   86436  100291  138200   81216  140477
River Rch & RM=Trinity River,1               ,181750
   50100   73271   85833   98659  132968   80854  134862
River Rch & RM=Trinity River,1               ,179572
   50100   73264   85552   97745  129718   80687  131451
River Rch & RM=Trinity River,1               ,178698
   50100   73264   85343   97119  127830   80562  129511
River Rch & RM=Trinity River,1               ,176021
   44300   64464   75864   85208  107043   73662  104979
River Rch & RM=Trinity River,1               ,172483
   44300   64464   75506   84264  104285   73418  102211
River Rch & RM=Trinity River,1               ,169025
   44300   64333   74951   83032  100582   72978   98662
River Rch & RM=Trinity River,1               ,167085
   44300   64040   74126   81420   96746   72288   94909
River Rch & RM=Trinity River,1               ,165454
   44300   63853   73493   80056   93413   71803   91647
River Rch & RM=Trinity River,1               ,165204
   44300   63853   73493   80056   93413   71803   91647
River Rch & RM=Trinity River,1               ,164199
   44300   63851   73372   79708   92019   71723   90329
River Rch & RM=Trinity River,1               ,162832
   44300   63848   73304   79382   90383   71680   88788
River Rch & RM=Trinity River,1               ,161707
   44300   63744   72732   78205   87601   71238   86073
River Rch & RM=Trinity River,1               ,159456
   44300   63597   71853   76383   83295   70567   81877
River Rch & RM=Trinity River,1               ,157344
   44300   63560   71536   75613   80665   70328   79284
River Rch & RM=Trinity River,1               ,154267
   44700   64260   72098   75896   79419   70858   78497
River Rch & RM=Trinity River,1               ,151264
   44700   64260   72095   75677   77074   70858   76106
River Rch & RM=Trinity River,1               ,148768
   44700   64260   72094   75646   76784   70858   75808
River Rch & RM=Trinity River,1               ,147333
   44700   66256   84088  101796  139875   79117  142868
River Rch & RM=Trinity River,1               ,145717
   44700   66228   83478  100066  134896   78712  137782
River Rch & RM=Trinity River,1               ,143893
   44700   66210   82907   98353  130099   78365  132907
River Rch & RM=Trinity River,1               ,141890
   44700   66207   82210   96461  125161   77933  127939
River Rch & RM=Trinity River,1               ,139225
   44700   66193   81673   95114  121844   77576  124666
River Rch & RM=Trinity River,1               ,137179
   44700   66182   81303   94221  119519   77320  122422
River Rch & RM=Trinity River,1               ,135104
   44700   66070   80442   92323  114967   76661  118012
River Rch & RM=Trinity River,1               ,133245
   44700   66070   80212   91574  112562   76521  115753
River Rch & RM=Trinity River,1               ,131382
   44700   66070   80113   91110  110670   76464  114010
River Rch & RM=Trinity River,1               ,129561
   44700   66049   79722   89961  107630   76194  111103
River Rch & RM=Trinity River,1               ,127110
   44700   65815   78807   88212  104089   75429  107679
River Rch & RM=Trinity River,1               ,124996
   44700   65743   78512   87518  102003   75176  105712
River Rch & RM=Trinity River,1               ,123554
   44700   65742   78271   86865  100204   74991  104042
River Rch & RM=Trinity River,1               ,122155
   44700   65729   78023   86289   98891   74783  102800
River Rch & RM=Trinity River,1               ,120905
   44700   65695   77673   85471   97034   74485  101039
River Rch & RM=Trinity River,1               ,118211
   44700   65695   77587   85149   95921   74416  100001
River Rch & RM=Trinity River,1               ,116211
   44700   65695   77575   85099   95457   74405   99637
River Rch & RM=Trinity River,1               ,113969
   40000   61295   71398   80343   87595   72241   88631
River Rch & RM=Trinity River,1               ,112556
   40000   61291   71281   79867   85924   72142   87038
River Rch & RM=Trinity River,1               ,110130
   40000   61291   71269   79694   85126   72132   86276
River Rch & RM=Trinity River,1               ,108725
   40000   61291   71269   79650   84751   72132   85924
River Rch & RM=Trinity River,1               ,107532
   40000   61291   71262   79394   83402   72131   84529
River Rch & RM=Trinity River,1               ,104348
   40000   62008   73422   84781  106737   73589  109056
River Rch & RM=Trinity River,1               ,96265
   40000   62005   73273   83325   99225   73526  101078
River Rch & RM=Trinity River,1               ,95077
   40000   62005   73246   82957   97670   73518   99415
River Rch & RM=Trinity River,1               ,91978
   40000   62000   73037   82047   94619   73393   96168
River Rch & RM=Trinity River,1               ,83613
   56100   86900  111100  141000  217800  104500  221300
River Rch & RM=Trinity River,1               ,80593
   56100   86900  111100  141000  217800  104500  221300
River Rch & RM=Trinity River,1               ,76398
   56100   86900  111100  141000  217800  104500  221300
River Rch & RM=Trinity River,1               ,74608
   56100   86900  111100  141000  217800  104500  221300
River Rch & RM=Trinity River,1               ,72672
   56100   86900  111100  141000  217800  104500  221300
River Rch & RM=Trinity River,1               ,71053
   56100   86900  111100  141000  217800  104500  221300
River Rch & RM=Trinity River,1               ,68028
   56100   86900  111100  141000  217800  104500  221300
River Rch & RM=Trinity River,1               ,65984
   56100   86900  111100  141000  217800  104500  221300
River Rch & RM=Trinity River,1               ,64637
   56100   86900  111100  141000  217800  104500  221300
River Rch & RM=Trinity River,1               ,62238
   56100   86900  111100  141000  217800  104500  221300
River Rch & RM=Trinity River,1               ,59702
   56100   86900  111100  141000  217800  104500  221300
River Rch & RM=Trinity River,1               ,56823
   56100   86900  111100  141000  217800  104500  221300
River Rch & RM=Trinity River,1               ,55303
   56100   86800  103899  118888  151146   99098  153198
River Rch & RM=Trinity River,1               ,53117
   56100   86875  109244  131796  181011  103218  183863
River Rch & RM=Trinity River,1               ,51036
   56100   86875  109005  130576  176441  103046  179203
River Rch & RM=Trinity River,1               ,48916
   51600   78575  102701  126168  167459  100774  168767
River Rch & RM=Trinity River,1               ,46568
   51600   78575  102301  123596  159545  100474  160751
River Rch & RM=Trinity River,1               ,45073
   51600   78575  101772  121544  154452  100036  155579
River Rch & RM=Trinity River,1               ,44793
   51600   78575  101772  121544  154452  100036  155579
River Rch & RM=Trinity River,1               ,43746
   51600   78575  101397  120399  151548   99708  152598
River Rch & RM=Trinity River,1               ,42372
   51600   78403   99736  117205  145757   98179  146712
River Rch & RM=Trinity River,1               ,39787
   51600   78400   99218  115868  142484   97711  143359
River Rch & RM=Trinity River,1               ,38724
   51600   78375   98359  113963  138763   96928  139570
River Rch & RM=Trinity River,1               ,37337
   51600   78266   97508  112342  135723   96140  136463
River Rch & RM=Trinity River,1               ,35159
   51600   77976   96109  109477  130089   94854  130684
River Rch & RM=Trinity River,1               ,32786
   51600   77976   96085  109217  128917   94838  129436
River Rch & RM=Trinity River,1               ,30239
   51600   77976   95951  108396  126459   94736  126840
River Rch & RM=Trinity River,1               ,28041
   51600   77976   95899  107960  124932   94696  125230
River Rch & RM=Trinity River,1               ,26191
   51600   77975   95621  106827  121908   94467  122064
River Rch & RM=Trinity River,1               ,24046
   51600   77975   95591  106502  120583   94451  120641
River Rch & RM=Trinity River,1               ,19761
   51600   77975   95591  106502  120357   94451  120374
River Rch & RM=Trinity River,1               ,17358
   51600   77975   95488  105875  118183   94379  118115
River Rch & RM=Trinity River,1               ,15600
   51600   77975   95488  105768  116821   94379  116665
River Rch & RM=Trinity River,1               ,13539
   51600   77975   95488  105742  116296   94379  116118
River Rch & RM=Trinity River,1               ,11371
   51600   78600  104501  133942  196620  102015  198170
River Rch & RM=Trinity River,1               ,9505
   51600   78600  104500  133677  195527  102015  197064
River Rch & RM=Trinity River,1               ,7604
   51600   78600  104500  133585  194701  102015  196225
River Rch & RM=Trinity River,1               ,6288
   51600   78600  104500  133542  194157  102015  195673
Boundary for River Rch & Prof#=Trinity River,1               , 1
Up Type= 0
Dn Type= 1
Dn Known WS=322.4
Boundary for River Rch & Prof#=Trinity River,1               , 2
Up Type= 0
Dn Type= 1
Dn Known WS=325.55
Boundary for River Rch & Prof#=Trinity River,1               , 3
Up Type= 0
Dn Type= 1
Dn Known WS=327.49
Boundary for River Rch & Prof#=Trinity River,1               , 4
Up Type= 0
Dn Type= 1
Dn Known WS=329.3
Boundary for River Rch & Prof#=Trinity River,1               , 5
Up Type= 0
Dn Type= 1
Dn Known WS=332.4
Boundary for River Rch & Prof#=Trinity River,1               , 6
Up Type= 0
Dn Type= 1
Dn Known WS=327.32
Boundary for River Rch & Prof#=Trinity River,1               , 7
Up Type= 0
Dn Type= 1
Dn Known WS=332.47
DSS Import GetInterval= 0
DSS Import GetPeak= 0
DSS Import FillOption= 0

--- TR_FEMA.f07 (steady flow) ---

Flow Title=2020 Dal14Ell3 Reduced Discharges
Program Version=5.06
BEGIN FILE DESCRIPTION:
Full discharges through Dallas LID14/Ellis LID3 with reduced discharges elsewhere based on With Levee supplemental model that used lateral structures to represent levees
Boundary condition - Known WS based on With Levee supplemental model
END FILE DESCRIPTION:
Number of Profiles= 7
Profile Names=10yr,25yr,50yr,100yr,500yr,1PCT_MINUS,1PCT_PLUS
River Rch & RM=Trinity River,1               ,205777
   50100   75100   95700  120200  185200   87400  193600
River Rch & RM=Trinity River,1               ,200569
   50100   75091   94845  117604  177387   87001  184767
River Rch & RM=Trinity River,1               ,198513
   50100   75059   94005  115435  171504   86543  178140
River Rch & RM=Trinity River,1               ,196991
   50100   74828   93020  113486  167115   85860  173248
River Rch & RM=Trinity River,1               ,195872
   50100   74766   92518  112383  164541   85541  170364
River Rch & RM=Trinity River,1               ,194145
   50100   74649   91729  110743  160793   85020  166172
River Rch & RM=Trinity River,1               ,193094
   50100   74595   91432  110146  159532   84818  164766
River Rch & RM=Trinity River,1               ,191491
   50100   74516   90901  108900  156308   84476  160955
River Rch & RM=Trinity River,1               ,189380
   50100   74324   89988  106968  152250   83859  156278
River Rch & RM=Trinity River,1               ,187750
   50100   74041   88838  104741  148012   83042  151481
River Rch & RM=Trinity River,1               ,186516
   50100   73520   87326  102185  143688   81880  146553
River Rch & RM=Trinity River,1               ,186264
   50100   73520   87326  102185  143688   81880  146553
River Rch & RM=Trinity River,1               ,184503
   50100   73288   86436  100291  138200   81216  140477
River Rch & RM=Trinity River,1               ,181750
   50100   73271   85833   98659  132968   80854  134862
River Rch & RM=Trinity River,1               ,179572
   50100   73264   85552   97745  129718   80687  131451
River Rch & RM=Trinity River,1               ,178698
   50100   73264   85343   97119  127830   80562  129511
River Rch & RM=Trinity River,1               ,176021
   44300   64464   75864   85208  107043   73662  104979
River Rch & RM=Trinity River,1               ,172483
   44300   64464   75506   84264  104285   73418  102211
River Rch & RM=Trinity River,1               ,169025
   44300   64333   74951   83032  100582   72978   98662
River Rch & RM=Trinity River,1               ,167085
   44300   64040   74126   81420   96746   72288   94909
River Rch & RM=Trinity River,1               ,165454
   44300   63853   73493   80056   93413   71803   91647
River Rch & RM=Trinity River,1               ,165204
   44300   63853   73493   80056   93413   71803   91647
River Rch & RM=Trinity River,1               ,164199
   44300   63851   73372   79708   92019   71723   90329
River Rch & RM=Trinity River,1               ,162832
   44300   63848   73304   79382   90383   71680   88788
River Rch & RM=Trinity River,1               ,161707
   44300   63744   72732   78205   87601   71238   86073
River Rch & RM=Trinity River,1               ,159456
   44300   63597   71853   76383   83295   70567   81877
River Rch & RM=Trinity River,1               ,157344
   44300   63560   71536   75613   80665   70328   79284
River Rch & RM=Trinity River,1               ,154267
   44700   64260   72098   75896   79419   70858   78497
River Rch & RM=Trinity River,1               ,151264
   44700   64260   72095   75677   77074   70858   76106
River Rch & RM=Trinity River,1               ,148768
   44700   67000   87100  109800  167700   81200  172800
River Rch & RM=Trinity River,1               ,147333
   44700   67000   87100  109800  167700   81200  172800
River Rch & RM=Trinity River,1               ,145717
   44700   67000   87100  109800  167700   81200  172800
River Rch & RM=Trinity River,1               ,143893
   44700   67000   87100  109800  167700   81200  172800
River Rch & RM=Trinity River,1               ,141890
   44700   67000   87100  109800  167700   81200  172800
River Rch & RM=Trinity River,1               ,139225
   44700   67000   87100  109800  167700   81200  172800
River Rch & RM=Trinity River,1               ,137179
   44700   67000   87100  109800  167700   81200  172800
River Rch & RM=Trinity River,1               ,135104
   44700   67000   87100  109800  167700   81200  172800
River Rch & RM=Trinity River,1               ,133245
   44700   67000   87100  109800  167700   81200  172800
River Rch & RM=Trinity River,1               ,131382
   44700   67000   87100  109800  167700   81200  172800
River Rch & RM=Trinity River,1               ,129561
   44700   67000   87100  109800  167700   81200  172800
River Rch & RM=Trinity River,1               ,127110
   44700   67000   87100  109800  167700   81200  172800
River Rch & RM=Trinity River,1               ,124996
   44700   67000   87100  109800  167700   81200  172800
River Rch & RM=Trinity River,1               ,123554
   44700   67000   87100  109800  167700   81200  172800
River Rch & RM=Trinity River,1               ,122155
   44700   67000   87100  109800  167700   81200  172800
River Rch & RM=Trinity River,1               ,120905
   44700   67000   87100  109800  167700   81200  172800
River Rch & RM=Trinity River,1               ,118211
   44700   67000   87100  109800  167700   81200  172800
River Rch & RM=Trinity River,1               ,116211
   44700   67000   87100  109800  167700   81200  172800
River Rch & RM=Trinity River,1               ,113969
   40000   62600   81000  105400  160900   79100  162800
River Rch & RM=Trinity River,1               ,112556
   40000   62600   81000  105400  160900   79100  162800
River Rch & RM=Trinity River,1               ,110130
   40000   62600   81000  105400  160900   79100  162800
River Rch & RM=Trinity River,1               ,108725
   40000   62600   81000  105400  160900   79100  162800
River Rch & RM=Trinity River,1               ,107532
   40000   62600   81000  105400  160900   79100  162800
River Rch & RM=Trinity River,1               ,104348
   40000   62600   81000  105400  160900   79100  162800
River Rch & RM=Trinity River,1               ,96265
   40000   62600   81000  105400  160900   79100  162800
River Rch & RM=Trinity River,1               ,95077
   40000   62600   81000  105400  160900   79100  162800
River Rch & RM=Trinity River,1               ,91978
   40000   62600   81000  105400  160900   79100  162800
River Rch & RM=Trinity River,1               ,83613
   56100   86900  111100  141000  217800  104500  221300
River Rch & RM=Trinity River,1               ,80593
   56100   86900  111100  141000  217800  104500  221300
River Rch & RM=Trinity River,1               ,76398
   56100   86297  102909  117395  153572   98669  156563
River Rch & RM=Trinity River,1               ,74608
   56100   86900  110479  138421  209309  104114  212555
River Rch & RM=Trinity River,1               ,72672
   56100   86896  109963  137070  205824  103731  208981
River Rch & RM=Trinity River,1               ,71053
   56100   86861  109210  135335  201676  103136  204734
River Rch & RM=Trinity River,1               ,68028
   56100   86838  108124  132522  192141  102287  194934
River Rch & RM=Trinity River,1               ,65984
   56100   86836  107011  129170  182626  101459  185223
River Rch & RM=Trinity River,1               ,64637
   56100   86834  106583  127365  176781  101167  179271
River Rch & RM=Trinity River,1               ,62238
   56100   86831  105966  125051  169878  100728  172248
River Rch & RM=Trinity River,1               ,59702
   56100   86800  104338  120222  156737   99453  158935
River Rch & RM=Trinity River,1               ,56823
   56100   86800  103899  118920  152495   99098  154591
River Rch & RM=Trinity River,1               ,55303
   56100   86800  103899  118888  151146   99098  153198
River Rch & RM=Trinity River,1               ,53117
   56100   86875  109244  131796  181011  103218  183863
River Rch & RM=Trinity River,1               ,51036
   56100   86875  109005  130576  176441  103046  179203
River Rch & RM=Trinity River,1               ,48916
   51600   78575  102701  126168  167459  100774  168767
River Rch & RM=Trinity River,1               ,46568
   51600   78575  102301  123596  159545  100474  160751
River Rch & RM=Trinity River,1               ,45073
   51600   78575  101772  121544  154452  100036  155579
River Rch & RM=Trinity River,1               ,44793
   51600   78575  101772  121544  154452  100036  155579
River Rch & RM=Trinity River,1               ,43746
   51600   78575  101397  120399  151548   99708  152598
River Rch & RM=Trinity River,1               ,42372
   51600   78403   99736  117205  145757   98179  146712
River Rch & RM=Trinity River,1               ,39787
   51600   78400   99218  115868  142484   97711  143359
River Rch & RM=Trinity River,1               ,38724
   51600   78375   98359  113963  138763   96928  139570
River Rch & RM=Trinity River,1               ,37337
   51600   78266   97508  112342  135723   96140  136463
River Rch & RM=Trinity River,1               ,35159
   51600   77976   96109  109477  130089   94854  130684
River Rch & RM=Trinity River,1               ,32786
   51600   77976   96085  109217  128917   94838  129436
River Rch & RM=Trinity River,1               ,30239
   51600   77976   95951  108396  126459   94736  126840
River Rch & RM=Trinity River,1               ,28041
   51600   77976   95899  107960  124932   94696  125230
River Rch & RM=Trinity River,1               ,26191
   51600   77975   95621  106827  121908   94467  122064
River Rch & RM=Trinity River,1               ,24046
   51600   77975   95591  106502  120583   94451  120641
River Rch & RM=Trinity River,1               ,19761
   51600   77975   95591  106502  120357   94451  120374
River Rch & RM=Trinity River,1               ,17358
   51600   77975   95488  105875  118183   94379  118115
River Rch & RM=Trinity River,1               ,15600
   51600   77975   95488  105768  116821   94379  116665
River Rch & RM=Trinity River,1               ,13539
   51600   77975   95488  105742  116296   94379  116118
River Rch & RM=Trinity River,1               ,11371
   51600   78600  104501  133942  196620  102015  198170
River Rch & RM=Trinity River,1               ,9505
   51600   78600  104500  133677  195527  102015  197064
River Rch & RM=Trinity River,1               ,7604
   51600   78600  104500  133585  194701  102015  196225
River Rch & RM=Trinity River,1               ,6288
   51600   78600  104500  133542  194157  102015  195673
Boundary for River Rch & Prof#=Trinity River,1               , 1
Up Type= 0
Dn Type= 1
Dn Known WS=322.4
Boundary for River Rch & Prof#=Trinity River,1               , 2
Up Type= 0
Dn Type= 1
Dn Known WS=325.55
Boundary for River Rch & Prof#=Trinity River,1               , 3
Up Type= 0
Dn Type= 1
Dn Known WS=327.49
Boundary for River Rch & Prof#=Trinity River,1               , 4
Up Type= 0
Dn Type= 1
Dn Known WS=329.3
Boundary for River Rch & Prof#=Trinity River,1               , 5
Up Type= 0
Dn Type= 1
Dn Known WS=332.4
Boundary for River Rch & Prof#=Trinity River,1               , 6
Up Type= 0
Dn Type= 1
Dn Known WS=327.32
Boundary for River Rch & Prof#=Trinity River,1               , 7
Up Type= 0
Dn Type= 1
Dn Known WS=332.47
DSS Import GetInterval= 0
DSS Import GetPeak= 0
DSS Import FillOption= 0
